HEC-RAS study LIKANARV.prj: LIKANARV

--- LIKANARV.g01 (geometry) --- (continued)

Type RM Length L Ch R = 1 ,44644   ,330.2,346.7,336.2
XS GIS Cut Line= 4
2159713.66885881662314.5128345322159794.92206267662447.943002655
2159819.35293076662620.2143066552159899.52987995662936.973810702
#Sta/Elev= 30
       0 1620.67    12.5 1618.24    45.3 1605.47    54.6 1600.65    67.8 1597.37
    82.7 1589.59    92.1 1587.71   105.6 1583.28   165.6 1569.15   169.6 1567.86
   177.7 1562.45   181.7  1561.1   189.8 1561.01   197.9  1558.5  214.391557.372
   226.2 1555.96  276.481557.371   286.8  1560.1   323.1  1564.3   384.4 1562.78
   413.7 1564.84   438.5  1564.6   492.1 1568.02   496.3 1568.96   504.5 1573.39
   512.7 1574.84     587 1582.75   611.8 1589.92   636.5 1599.96     657 1599.89
#Mann= 4 ,-1,0
       0      .1       0  214.39    .045       0  276.48      .1       0
  580.22     .06       0
Bank Sta=214.39,276.48
XS Rating Curve= 0 ,0
Exp/Cntr=0.3,0.1

Type RM Length L Ch R = 1 ,44297   ,262.9,254.2,235.2
XS GIS Cut Line= 4
2159443.34588534662354.644989208 2159479.1337749662475.903423968
2159498.00261871662706.4824932552159624.82342671662985.915730665
#Sta/Elev= 30
       0 1632.26    15.2 1628.01    31.7 1620.85    73.5 1596.72    86.4 1590.72
    96.1 1587.71   115.4 1584.78   127.7 1579.99   135.7 1578.63   163.8  1560.7
   179.9 1552.81   187.9 1552.15     216 1556.97  233.72 1551.48   244.1 1549.97
   288.2 1550.09  296.05 1551.48   308.3  1553.4   324.4 1558.97   354.9 1561.45
   373.9 1560.25   387.1 1562.16   404.7 1560.65     431 1564.22   508.2 1567.39
   537.3  1574.3   611.1 1584.28   624.3 1587.56   642.4 1587.16   664.6 1594.92
#Mann= 4 ,-1,0
       0      .1       0  233.72    .045       0  296.05      .1       0
  637.78     .06       0
Bank Sta=233.72,296.05
XS Rating Curve= 0 ,0
Exp/Cntr=0.3,0.1

Type RM Length L Ch R = 1 ,44043   ,234.4,243,253.9
XS GIS Cut Line= 3
2159201.60755713662439.8451572642159232.69917869662601.348858107
2159504.75086727663004.676282137
#Sta/Elev= 30
       0 1599.28    25.8 1591.63    46.2 1587.76    62.5    1589    74.1 1586.57
    82.8 1586.17    99.1  1581.6   115.4 1580.34   127.6 1578.02   139.9 1574.85
   156.1 1568.58   169.1 1567.13   178.7 1560.36   193.2 1552.57  211.21 1549.56
   231.8 1547.17   253.3 1547.42   264.8 1549.53   270.4 1550.64   275.2 1553.22
   280.1 1554.42   322.4 1556.21   443.5 1556.47     502 1557.63   511.7 1559.41
   549.8 1569.72   593.7 1579.53   617.8 1587.26   630.7 1595.53     651 1593.17
#Mann= 4 ,-1,0
       0      .1       0  211.21    .045       0   264.8      .1       0
  624.47     .06       0
Bank Sta=211.21,264.8
XS Rating Curve= 0 ,0
Exp/Cntr(USF)=0,0
Exp/Cntr=0.3,0.1

Type RM Length L Ch R = 1 ,43800   ,582.1,575.5,555.3
XS GIS Cut Line= 4
2159040.80603192662488.2915705932159053.06723741662723.668616007
2159110.71410583662933.1385489662159331.93742671663162.254455935
#Sta/Elev= 30
       0 1596.31      49 1589.04      65 1587.34      73 1585.64      81 1585.81
      85 1585.16      93 1582.89   121.1 1577.48   153.1 1568.54   189.1 1565.18
   221.2 1559.73   233.2 1558.73   262.2 1552.78   270.5 1549.92   282.9  1547.7
   291.2 1545.99   328.5 1545.75     3441547.702   361.7 1550.12   415.7 1551.73
   441.2 1554.09   458.6 1557.24   468.2 1559.87   503.1 1562.79   675.4 1582.83
   725.5 1589.02   736.6    1591   753.3 1592.05   762.4 1594.18   771.4 1599.06
#Mann= 5 ,-1,0
       0      .1       0   282.9    .045       0     344      .1       0
  622.95     .06       0  762.95      .1       0
Bank Sta=282.9,344
XS Rating Curve= 0 ,0
Exp/Cntr=0.3,0.1

Type RM Length L Ch R = 1 ,43224   ,353.9,362,362.6
XS GIS Cut Line= 3
2158491.35898921662939.5972266182158709.74667716 663235.53796268
2158997.03239433663445.632090828
#Sta/Elev= 30
       0 1574.61    18.9 1568.34    55.3 1558.88   141.2 1553.06   176.5 1552.83
   205.8 1550.51  237.511540.984   250.5 1539.41   280.4 1539.75  285.981540.983
   296.3 1547.12   302.1 1548.62     335 1551.13   354.9 1550.59   442.3 1555.01
   544.2 1569.42   568.2 1569.22     574 1571.42   585.4 1579.69   591.1 1582.64
     594 1583.43   602.6 1582.31   611.2 1582.87   619.7  1586.5   633.4 1588.93
   648.3 1594.91   668.4  1599.5     697 1607.93   708.5 1609.96   723.7 1616.02
#Mann= 6 ,-1,0
       0     .06       0      20      .1       0  237.51    .045       0
  285.98      .1       0   477.8     .06       0  723.71      .1       0
Bank Sta=237.51,285.98
XS Rating Curve= 0 ,0
Exp/Cntr=0.3,0.1

Type RM Length L Ch R = 1 ,42862   ,383.8,389.9,381.1
XS GIS Cut Line= 3
2158259.08030665 663090.765949192158397.80941862663440.431029226
2158429.22888804663776.360647931
#Sta/Elev= 30
       0 1577.39     6.9 1576.59    24.1  1570.2    41.3  1570.2    49.9 1571.65
    58.5 1571.42    84.4 1564.43   123.1 1556.99     136 1557.15   147.5 1553.79
   170.4 1549.41  195.98 1537.26   200.5  1535.6   217.8 1535.14   247.9 1535.33
  258.171537.257   269.4 1540.18   290.9 1543.28   304.6  1543.4   329.6 1545.98
   437.2 1547.45   449.2 1548.54   497.5 1548.22     515 1548.89   533.6 1551.51
   561.7 1551.84   587.1 1558.46   606.8 1561.85     634 1568.15   713.6 1592.83
#Mann= 5 ,-1,0
       0      .1       0  195.98    .045       0  258.17      .1       0
  486.18     .06       0  586.18      .1       0
Bank Sta=195.98,258.17
XS Rating Curve= 0 ,0
Exp/Cntr=0.3,0.1

Type RM Length L Ch R = 1 ,42472   ,361.9,373,378.9
XS GIS Cut Line= 4
 2157949.6391812663178.1426506292157957.75790935663364.057983317
2158078.19664523663646.2343758992158079.46797859663903.529641588
#Sta/Elev= 30
       0 1587.16      11 1585.43    23.1 1580.82    31.1 1580.56    43.1 1577.76
    75.1 1572.72   119.1 1562.76   183.2 1554.94   187.3 1553.78   191.7 1549.61
     196    1544   200.4 1541.37   249.8 1540.27  267.88    1535   274.3 1533.56
   298.5 1533.08   310.7 1533.19  320.621534.999   338.1 1538.95   356.4 1537.96
   383.9 1538.24     396 1539.44   409.1 1538.52   420.4 1539.89   492.9 1544.05
   515.8 1544.86   527.8 1551.18   543.8 1556.83   614.5 1573.67   750.2 1613.85
#Mann= 5 ,-1,0
       0      .1       0  267.88    .045       0  320.62      .1       0
  386.09     .06       0   492.9      .1       0
Bank Sta=267.88,320.62
XS Rating Curve= 0 ,0
Exp/Cntr=0.3,0.1

Type RM Length L Ch R = 1 ,42099   ,356.5,367.1,374.9
XS GIS Cut Line= 4
2157759.15954563  663163.36072182157665.68192694663338.071888573
2157660.70340494663660.6253555152157586.53251531663800.288511319
#Sta/Elev= 30
       0  1589.8    33.8 1579.83      52 1575.46    74.6 1563.49   110.9  1560.5
   151.3 1550.77   174.5 1548.87   195.6 1543.71   229.3 1537.66   245.3 1536.18
   269.3 1535.79   429.3 1537.52  446.931531.894   453.3 1530.45   473.3 1529.37
   481.3 1529.88  486.641531.895   489.3 1533.88   493.3 1538.55   497.3    1541
   525.9 1542.76   530.4 1544.95   539.3 1554.68     544 1558.76   548.5 1561.88
   557.6 1565.46   571.2  1576.5   604.4  1593.3   643.7 1616.47   678.9 1638.62
#Mann= 7 ,-1,0
       0     .06       0     100     .07       0  208.15      .1       0
  408.15     .06       0  446.93    .045       0  486.64     .06       0
  508.15      .1       0
Bank Sta=446.93,486.64
XS Rating Curve= 0 ,0
Exp/Cntr=0.3,0.1

Type RM Length L Ch R = 1 ,41732   ,189.9,197.1,194.6
XS GIS Cut Line= 3
2157551.04158111663053.5573909992157278.50241571663559.004102029
2157288.36165843663739.737870082
#Sta/Elev= 30
       0  1588.6    39.8 1577.15    72.3 1566.06    90.4 1561.47   190.4  1545.7
   235.9 1544.12   263.1 1539.75   317.7 1537.47   363.1 1530.72   390.4 1529.77
     404 1530.82   431.3 1528.69   438.8 1526.93   449.5 1528.64   455.5 1527.11
   469.6 1525.88   494.9 1527.12   522.2 1526.87   530.3 1529.81   540.4  1537.8
   572.2 1538.42   580.4  1542.8   588.4  1544.7   592.4 1549.25   600.5 1561.42
   604.4 1563.98   640.5 1574.12   668.6 1586.35   724.6 1615.04   755.2 1624.23
#Mann= 7 ,-1,0
       0      .1       0     110     .06       0     280      .1       0
     450     .06       0   455.5    .045       0   494.9     .06       0
     560      .1       0
Bank Sta=455.5,494.9
XS Rating Curve= 0 ,0
Exp/Cntr=0.3,0.1

Type RM Length L Ch R = 1 ,41535   ,68.7,70.5,75
XS GIS Cut Line= 4
2157434.70163372662975.9503168582157256.06101394663267.802771228
2157100.70125267 663474.658258572157056.05127867663715.922893728
#Sta/Elev= 30
       0 1592.31    29.6 1585.68    81.3 1570.92   127.4 1555.75   170.3 1549.51
   181.1 1545.51   191.8 1545.12   204.1 1547.52   217.2  1541.7   229.6 1540.18
   254.7 1542.87   268.8 1535.36   273.5 1534.57   353.9 1530.82  392.28 1523.26
   408.6 1520.88   435.2 1523.21   451.6 1521.85   471.6 1527.13     519 1527.16
   535.2 1530.56   561.8  1528.4   611.6 1528.71   652.3 1533.21   660.4 1535.92
   705.1 1543.54   778.4 1553.26   802.8 1560.99     815 1559.51   846.2  1563.7
#Mann= 11 ,-1,0
       0      .1       0      90     .06       0     210     .08       0
     220     .06       0     320     .08       0  392.28    .045       0
   435.2     .05       0  442.18     .06       0  572.18     .05       0
  670.88     .06       0  780.88      .1       0
Bank Sta=392.28,435.2
XS Rating Curve= 0 ,0
Exp/Cntr=0.3,0.1

Type RM Length L Ch R = 1 ,41464   ,103.4,104.2,104.3
XS GIS Cut Line= 4
2157358.30653602662964.1991474442157179.66591625663256.051601814
2157052.07498309663423.8577703032156994.65788838663678.365678425
#Sta/Elev= 30
       0  1583.1    29.3 1573.87    77.9 1560.66   109.9 1554.35   188.7 1535.49
   249.5 1530.74   301.9 1528.36   345.5 1528.25   350.8 1527.04   359.8 1523.08
   368.7 1520.75   376.9 1519.89   408.9 1519.33     419 1520.42  428.46 1523.06
   439.1 1525.64   449.1 1526.58   493.9 1524.79   519.8 1525.48   536.7  1522.4
     551 1524.14   558.4 1526.41   570.7 1526.94   578.9 1524.45   587.1 1523.99
   607.8 1528.09   679.8  1534.7   694.5 1539.22   726.6 1540.98   813.9 1542.73
#Mann= 9 ,-1,0
       0      .1       0      80     .06       0     270     .05       0
   359.8    .045       0  428.46     .05       0  462.18     .06       0
  582.99     .05       0  682.99     .06       0  782.99     .07       0
Bank Sta=359.8,428.46
XS Rating Curve= 0 ,0
Exp/Cntr=0.3,0.1

Type RM Length L Ch R = 1 ,41360   ,306.3,309.2,313.4
XS GIS Cut Line= 4
 2157278.8058499662963.0323474042156926.94593521663417.962338114
2156820.32171864663385.9750731432156642.61469101663575.529235939
#Sta/Elev= 30
       0 1576.93    58.3 1554.58   114.6 1541.52   169.6 1531.37   191.6 1529.15
   245.4 1526.72   260.6 1527.13   285.9  1522.8   305.7  1521.8   318.1 1518.74
   331.3    1518   350.8 1518.63  362.32 1521.79   376.9 1524.84     394 1523.49
   416.2 1523.64   442.4  1525.9   548.8 1528.78   553.9 1529.36   559.4 1531.93
   574.1 1533.79   590.5 1533.56   633.5 1529.91   793.5 1531.78     806 1534.69
     836 1535.42   855.8 1538.72   891.4  1545.6   906.7 1552.27   946.3 1554.37
#Mann= 7 ,-1,0
       0     .06       0     240     .05       0   305.7    .045       0
  362.32     .05       0     420     .08       0     490     .06       0
  906.44      .1       0
Bank Sta=305.7,362.32
XS Rating Curve= 0 ,0
Exp/Cntr(USF)=0,0
Exp/Cntr=0.3,0.1

Type RM Length L Ch R = 1 ,41051   ,433.5,443.9,440.5
XS GIS Cut Line= 3
2157036.47769275662826.6660399612156626.06988817663240.229338563
2156407.75201362663329.240491084
#Sta/Elev= 30
       0 1578.86    40.2 1564.11    51.5 1557.17    62.9  1555.5   103.8 1537.97
   165.1  1529.4   178.2 1524.94   204.9 1523.63  211.62 1520.85   223.3 1516.73
   250.9 1515.76   261.6 1517.09266.27981520.851   273.5  1523.9   381.1 1519.34
   414.9 1522.59   482.5 1519.88   528.1  1520.2   542.2 1526.85   584.4 1535.36
   610.6 1547.12   621.6 1548.49   653.8 1547.92   658.1 1549.26   688.4 1576.02
   727.2 1601.79   766.1 1620.08   774.8  1622.6   796.6  1625.9   818.4 1626.38
#Mann= 9 ,-1,0
       0      .1       0      40     .06       0     160     .07       0
     180      .1       0  211.62    .045       0266.2798      .1       0
     320     .05       0     440     .06       0     580      .1       0
Bank Sta=211.62,266.2798
XS Rating Curve= 0 ,0
Exp/Cntr=0.3,0.1

Type RM Length L Ch R = 1 ,40607   ,550.6,560.9,555.4
XS GIS Cut Line= 3
2156719.21108593662571.4733790962156391.15052738662882.025138987
 2156296.4448694663105.225273779
#Sta/Elev= 30
       0 1562.51    14.7 1556.82      26 1551.18      49 1548.77    68.4 1544.29
    92.3 1540.72    99.6 1537.93   114.3 1528.97   136.4 1528.16   152.9 1521.85
   182.9 1521.27   226.9 1522.79   238.2 1520.95   263.7 1516.51   280.6 1516.28
   286.3 1516.54   294.8 1519.92  301.121521.053   312.6 1525.98   362.7 1527.55
   389.7 1530.34   422.1 1532.04   450.5 1539.23     490 1539.47   537.7 1542.21
   559.4 1548.41   602.9 1556.95   623.2 1562.05   659.4 1565.77   694.2 1576.41
#Mann= 5 ,-1,0
       0     .06       0     130      .1       0   238.2    .045       0
  301.12     .07       0     420      .1       0
Bank Sta=238.2,301.12
XS Rating Curve= 0 ,0
Exp/Cntr=0.3,0.1

Type RM Length L Ch R = 1 ,40046   ,650,684.5,675.3
XS GIS Cut Line= 3
2156286.41705476662231.4791389872156007.04269335662565.160525678
2155833.66208593662752.642630995
#Sta/Elev= 30
       0 1554.95     8.5 1553.56      16    1551    25.5 1549.67      70 1536.64
    75.3 1533.92    85.7 1525.32    90.8 1524.16   101.3 1523.53  108.471520.322
   133.4 1516.19   137.9 1516.74   143.1 1519.24   148.3 1520.27   173.2 1521.03
   221.6 1520.32   257.8 1524.43     389 1529.33   400.3 1531.24   445.3 1530.74
     457 1532.91   502.3 1536.99   527.8 1541.16     566 1542.07   590.1 1547.89
   601.4 1552.86   610.3 1554.73   636.8  1564.8   672.2 1572.99   690.6 1578.16
#Mann= 8 ,-1,0
       0     .06       0      80      .1       0  108.47    .045       0
   148.3      .1       0     180     .05       0     230     .07       0
     300     .06       0     390      .1       0
Bank Sta=108.47,148.3
XS Rating Curve= 0 ,0
Exp/Cntr=0.3,0.1

Type RM Length L Ch R = 1 ,39362   ,475.9,543.7,555
XS GIS Cut Line= 4
2155939.81993345 661933.642974722155703.95503707661981.168460832
 2155552.6016767662127.0794138282155339.43661501662357.117417866
#Sta/Elev= 30
       0 1566.66    53.6 1562.94   105.7 1560.64   138.5 1557.33   186.1 1547.34
     237 1533.25   262.5 1528.52   290.3 1526.65   301.4  1520.2   322.5 1520.81
  329.921519.554   338.6 1517.94   373.2 1516.01   378.9 1517.28  382.141519.551
   390.3 1523.77   404.5 1526.82   463.2 1528.97   475.5 1538.15   486.8 1540.09
   491.9  1542.4   500.7 1548.37   519.1 1554.25   580.9 1560.34   644.6 1561.97
   655.5  1563.1   676.2 1570.94   715.9 1579.97   733.9 1586.19   764.5 1598.89
#Mann= 5 ,-1,0
       0      .1       0     100     .06       0  329.92    .045       0
  382.14     .05       0  610.84      .1       0
Bank Sta=329.92,382.14
XS Rating Curve= 0 ,0
Exp/Cntr=0.3,0.1

Type RM Length L Ch R = 1 ,38818   ,671.5,681.4,676.3
XS GIS Cut Line= 3
2155953.62255266661889.1525450632155745.00977758 661762.00433783
2155343.30511541661538.172288969
#Sta/Elev= 30
       0 1566.23   217.2 1557.49   230.5 1554.94   245.3 1553.98   260.2 1550.75
   324.9 1531.75   352.8 1525.58   378.1 1523.25   423.8 1522.33  432.981518.491
   443.2 1515.12   460.2 1514.47     472 1515.03  480.111518.489   492.5 1521.84
   504.3 1529.08   510.8 1531.33   527.8 1534.44   556.6 1534.51   561.2 1535.79
   565.8 1540.75   574.7 1556.35   580.8 1562.75   593.3 1569.95   620.7 1582.79
   629.9 1585.02     662 1604.02   671.1 1608.43   689.4 1620.94   704.2 1629.25
#Mann= 7 ,-1,0
       0      .1       0      40     .05       0     130      .1       0
     230     .06       0  432.98    .045       0  480.11     .06       0
  584.31      .1       0
Bank Sta=432.98,480.11
XS Rating Curve= 0 ,0
Exp/Cntr=0.3,0.1

Type RM Length L Ch R = 1 ,38136   ,503.9,493.7,465.5
XS GIS Cut Line= 4
2156342.81504886 661152.395976422156086.00406065661216.836017685
2155863.27302462661061.6594383132155691.03722662661054.227722821
#Sta/Elev= 30
       0 1585.74    93.5 1561.58   105.8 1559.51   118.2 1555.34   159.4 1544.83
   192.4 1543.39   208.9 1539.18   254.3  1532.8   325.5 1524.91   354.8 1522.83
   376.1 1518.47   403.8 1518.55  412.151517.519   418.2  1515.4   452.3 1513.88
  466.791517.517   484.2 1523.38   498.6 1525.13   510.8 1529.65   520.5 1536.08
   525.4 1537.49   539.7 1538.57   567.4 1536.53   571.4 1537.41   595.4 1556.31
   607.4 1560.44   631.8  1571.3   679.5 1594.83   691.5 1597.83   708.6 1608.04
#Mann= 7 ,-1,0
       0      .1       0     110     .06       0     120      .1       0
  334.77     .06       0  412.15    .045       0  466.79     .06       0
  556.23      .1       0
Bank Sta=412.15,466.79
XS Rating Curve= 0 ,0
Exp/Cntr=0.3,0.1

Type RM Length L Ch R = 1 ,37643   ,466.1,470.6,476.8
XS GIS Cut Line= 3
     2156498.017      660674.096     2156088.749      660687.851
      2155679.48      660701.607
#Sta/Elev= 30
       0 1715.98     9.8 1712.77    33.9 1695.07    93.9 1656.62   105.9 1649.94
   121.9  1638.3   133.9 1627.36   145.9 1624.44   165.9 1610.03   181.9 1600.66
   217.7 1583.15     234 1579.86   244.8 1574.69     270  1565.5   342.5 1535.57
     354 1526.97   374.1 1525.55  387.661516.852   394.1 1513.78   402.1 1513.62
   434.1 1513.63     4441516.853   570.2 1529.32   578.2 1531.18   590.2  1537.4
   594.2 1538.08   677.9 1540.76   742.3 1549.35   763.7 1550.47     819 1557.41
#Mann= 9 ,-1,0
       0      .1       0     170     .06       0     270     .05       0
     360     .06       0  387.66    .045       0     444     .06       0
   449.5     .05       0   459.5     .06       0   559.5      .1       0
Bank Sta=387.66,444
XS Rating Curve= 0 ,0
Exp/Cntr=0.3,0.1

Type RM Length L Ch R = 1 ,37172   ,594.9,599.4,604.6
XS GIS Cut Line= 4
2156474.84190881660269.5049232472156154.46856156660228.049939209
2155917.59180052660193.328455513     2155693.406      660152.677
#Sta/Elev= 30
       0 1674.95    10.8  1671.7      43 1650.97    63.2 1640.08   138.4 1605.57
   168.1 1588.57   183.4 1585.15   200.3 1576.11   260.8 1552.94   272.9 1550.72
     281 1545.58   301.2 1537.27   309.2 1529.83   329.4 1527.42  353.391516.059
   361.7 1513.86     382 1513.42   406.2 1513.57  415.55 1516.06   447.5 1522.11
   515.4 1523.58   535.6 1529.75   551.8 1537.27   600.5 1539.33   624.9 1549.56
   653.3 1565.86     698 1581.22   710.2 1583.53   734.6 1596.48   790.3 1616.33
#Mann= 7 ,-1,0
       0      .1       0     150     .06       0  343.04     .05       0
  353.39    .045       0  415.55     .05       0  443.04     .06       0
  543.04      .1       0
Bank Sta=353.39,415.55
XS Rating Curve= 0 ,0
Exp/Cntr=0.3,0.1

Type RM Length L Ch R = 1 ,36573   ,681.7,680.6,662.9
XS GIS Cut Line= 4
2156465.38142401659810.8117743252156128.32006232659724.158697572
2155950.15746769 659624.909537532155724.11216794659624.173137545
#Sta/Elev= 30
       0 1569.82   120.6 1548.23   195.4 1540.64   211.9 1537.64   273.8 1530.85
   380.2 1520.83   407.7 1519.62   421.4 1514.72   444.1 1514.43  450.181512.256
   467.2 1510.91   494.4 1510.97  499.741512.254   517.6  1520.9   531.3 1533.11
   535.9 1535.33   565.6 1538.99   577.9 1539.66   589.9 1538.48   593.9 1539.36
   597.9 1542.12   602.4 1547.69   613.9 1565.15   617.9 1570.03   633.9 1581.75
   665.9 1598.84   705.9 1616.74   717.9 1620.28   753.9 1639.62     778 1656.46
#Mann= 7 ,-1,0
       0      .1       0     240     .06       0     340      .1       0
  388.02     .07       0  450.18    .045       0  499.74     .06       0
  561.96      .1       0
Bank Sta=450.18,499.74
XS Rating Curve= 0 ,0
Exp/Cntr=0.3,0.1

Type RM Length L Ch R = 1 ,35892   ,510.4,525.9,520.1
XS GIS Cut Line= 4
2156519.53142648659199.7750944342156350.91135862659069.230896544
2156056.14391177659000.3888565482155832.18662255659025.077076049
#Sta/Elev= 30
       0 1574.25    29.9 1569.66    34.6 1568.05    43.4 1561.73    49.8 1558.85
    69.8 1553.05   100.4 1550.66   174.1 1540.15   186.4  1536.9   201.5 1529.11
   224.3  1528.3  251.291508.534   257.1 1505.94   265.3 1505.47   306.4 1507.25
  312.031508.531   322.9 1512.81   343.4  1515.1   372.1 1515.26   384.5 1511.35
   388.6 1511.42   413.2 1517.79   433.8 1533.64     442 1537.28   499.5 1535.73
     532 1537.48   580.3 1536.57   664.8 1537.78   708.7 1545.79   741.3 1549.69
#Mann= 7 ,-1,0
       0      .1       0     110     .06       0  233.25      .1       0
  251.29    .045       0  312.03      .1       0  433.25     .07       0
  535.95      .1       0
Bank Sta=251.29,312.03
XS Rating Curve= 0 ,0
Exp/Cntr=0.3,0.1

Type RM Length L Ch R = 1 ,35366   ,507.4,502.1,481.1
XS GIS Cut Line= 4
2156718.36902471658831.041506972 2156487.8494962658641.880228772
2156322.49078353658542.0036384042156168.94078835       658430.93
#Sta/Elev= 30
       0 1571.32      37 1560.84    85.6 1551.08   122.3 1541.29   154.3 1534.25
   192.1 1522.79   223.6  1515.3     253 1512.29   356.7 1511.62   359.7 1511.16
   368.4 1506.32   391.3 1507.99  404.161504.882   412.1 1503.29     424 1502.94
   433.3 1503.21  441.32 1504.88   461.6  1510.4   480.1 1528.15   489.4 1533.71
   510.8 1536.15   533.7 1536.34   538.7 1538.07     561  1564.4   568.1 1568.92
   611.1    1585     634 1591.85   662.1  1602.5     672 1604.15   680.9 1607.88
#Mann= 5 ,-1,0
       0      .1       0     250     .06       0  404.16    .045       0
  441.32     .06       0  531.38      .1       0
Bank Sta=404.16,441.32
XS Rating Curve= 0 ,0
Exp/Cntr=0.3,0.1

Type RM Length L Ch R = 1 ,34864   ,429.4,421,393.7
XS GIS Cut Line= 4
2156977.33646831658422.6960215392156824.22983777658297.818619771
2156584.42937099658241.4849489132156370.78195057658103.022911915
#Sta/Elev= 30
       0  1582.7    27.7 1575.09    68.6    1552    73.8 1548.19    84.1 1535.34
    89.2 1533.28   115.1 1531.62   140.9 1527.84   151.2  1525.1   161.5 1520.29
   214.1 1511.24   226.4 1505.64   251.4 1503.26  259.231501.165   267.5 1498.54
   296.2 1498.36  320.031501.165   337.3 1506.23   352.5 1507.55   464.6 1511.29
   487.1  1514.8   501.4 1520.95   510.9 1521.58   520.5 1526.39   551.3 1526.36
   568.1 1539.04   596.7 1553.12   623.6 1562.97   649.2 1568.66   698.5 1586.79
#Mann= 7 ,-1,0
       0      .1       0      70     .06       0  197.58      .1       0
  259.23    .045       0  320.03      .1       0  397.58     .06       0
   513.9      .1       0
Bank Sta=259.23,320.03
XS Rating Curve= 0 ,0
Exp/Cntr=0.3,0.1

Type RM Length L Ch R = 1 ,34443   ,263.1,292.6,307
XS GIS Cut Line= 5
2157145.20017186657937.3741028232156840.11114995657782.327570533
2156789.73062654657857.8423623542156657.75382899657906.240459624
2156408.48907194657932.606501349
#Sta/Elev= 30
       0 1601.48    18.1 1595.09      46 1591.49    81.9 1583.09   167.5 1542.85
   194.1 1531.97   225.5 1521.39   256.9 1513.73   274.6  1510.7   324.2 1508.46
   451.7 1507.42     456 1506.43  463.98 1500.66   468.7 1497.71   483.8 1497.17
   514.7 1497.99     524 1500.68   557.8 1508.05   595.3 1508.86   619.4 1516.83
   651.6 1515.39   659.6 1516.77   679.7 1525.45   691.8  1533.8   707.9 1540.32
   752.1 1543.16   764.2 1549.72   776.3 1553.34   806.8 1574.04   824.2 1582.64
#Mann= 8 ,-1,0
       0      .1       0     250     .06       0  372.23     .05       0
  463.98    .045       0     524     .07       0  603.58      .1       0
  703.58     .08       0  803.58      .1       0
Bank Sta=463.98,524
XS Rating Curve= 0 ,0
Exp/Cntr=0.3,0.1

Type RM Length L Ch R = 1 ,34151   ,237.3,255.7,248.2
XS GIS Cut Line= 2
2157169.59953821657855.9420818722156483.65041159657479.203183315
#Sta/Elev= 30
       0 1590.19    63.9  1583.2    92.9 1565.06   112.1 1555.46   159.2 1535.13
   185.7 1525.57   238.7 1511.84     280 1508.47   324.2 1508.99   435.2 1503.13
   444.9 1500.24   508.2 1499.17   517.3  1496.4   549.3 1495.69   556.9 1499.17
   565.7 1506.69   571.6 1509.11   609.9 1513.24   617.7 1518.73   630.5 1530.89
   649.7 1542.98     660 1544.41   663.3 1544.54   672.5 1548.75   686.5 1549.11
   704.4 1561.42   727.2 1571.62   736.4 1573.28   754.2 1581.95   782.6 1588.94
#Mann= 9 ,-1,0
       0      .1       0      50     .06       0      60      .1       0
     280     .06       0     460     .07       0   508.2    .045       0
   556.9     .08       0     660      .1       0     730     .08       0
Bank Sta=508.2,556.9
XS Rating Curve= 0 ,0
Exp/Cntr(USF)=0,0
Exp/Cntr=0.3,0.1

Type RM Length L Ch R = 1 ,33895   ,250.4,225.7,223.9
XS GIS Cut Line= 3
2157213.72392266657760.8511892982156802.88277608657372.819810702
2156632.03487995657329.608642535
#Sta/Elev= 30
       0 1566.32    12.2  1561.5    29.2 1559.31    40.6 1554.53    80.1 1542.51
     116 1533.45   139.3 1526.23   222.2  1508.7   238.5 1507.44   255.5 1504.09
   331.9 1501.96   359.8 1502.48   366.5 1500.99   387.3 1500.63  427.071495.945
   442.3 1493.78   458.8 1493.03     483 1494.36  488.751495.945   510.2 1503.96
     547 1511.81   609.9 1510.76   613.2 1511.74     623 1518.84   629.6 1522.46
   645.2 1528.47   682.3 1540.17   695.8 1546.45   712.3 1549.39   741.3 1564.32
#Mann= 8 ,-1,0
       0     .06       0      40      .1       0     260     .06       0
  427.07    .045       0  488.75     .07       0     540     .08       0
  645.12      .1       0  695.12     .08       0
Bank Sta=427.07,488.75
XS Rating Curve= 0 ,0
Exp/Cntr=0.3,0.1

Type RM Length L Ch R = 1 ,33669   ,81.3,80.7,82.5
XS GIS Cut Line= 3
2157594.47794305657512.4787869122156864.13177224657242.077242723
2156680.83520268657212.302050874
#Sta/Elev= 30
       0 1535.93    49.4 1527.63     104 1521.83   126.2 1518.15   160.3 1515.75
   177.3 1512.11   211.5 1509.15   228.5 1509.81   249.8 1507.76     284 1507.23
   321.9 1503.36   356.5 1503.33   377.8 1500.58   401.2 1499.16     490 1498.64
  521.021495.686   539.8 1491.79   565.5 1491.23   580.2 1492.02  589.931495.684
     602 1500.54   611.4 1502.18   689.2 1505.06   778.8 1510.13   827.4 1509.24
   839.5 1516.77     918 1540.03   932.7 1547.18   944.9 1548.61   964.5 1554.59
#Mann= 9 ,-1,0
       0     .05       0      90      .1       0     400     .06       0
     490     .08       0  521.02    .045       0  589.93     .08       0
     720     .07       0   778.8     .06       0   818.8     .08       0
Bank Sta=521.02,589.93
XS Rating Curve= 0 ,0
Exp/Cntr=0.3,0.1

Type RM Length L Ch R = 1 ,33589   ,242.8,220.6,207.2
XS GIS Cut Line= 3
 2157623.8041458  657439.92694252156893.45797499657169.525398311
2156659.83264707657135.309433666
#Sta/Elev= 30
       0 1542.78    46.5 1527.79   101.5 1517.54   126.4 1510.61   169.2 1506.79
   195.8 1501.95   225.7 1501.71   281.1 1504.84   306.7 1503.44   370.7 1504.44
   481.2 1497.25   502.9  1491.9   541.3  1495.6   579.7 1491.44   596.8 1495.09
  610.071495.613     640 1497.14   656.5  1498.6   677.3 1506.14   686.3 1506.33
   699.1 1502.53   733.7 1502.72   767.4 1504.62   808.4 1510.59   840.7 1508.63
   848.8 1512.57   856.9 1517.16   966.1 1547.46   982.2 1548.87  1014.9 1559.94
#Mann= 11 ,-1,0
       0     .05       0      10     .06       0     120     .05       0
     220      .1       0     290     .08       0   541.3    .045       0
  610.07     .03       0     640     .08       0     750     .06       0
   848.8     .08       0   948.8      .1       0
#XS Ineff= 2 , 0
                          684.17         1518.76
Permanent Ineff=
       F       F
Bank Sta=541.3,610.07
XS Rating Curve= 0 ,0
Exp/Cntr=0.3,0.1

Type RM Length L Ch R = 1 ,33368   ,693.1,656.1,639.8
XS GIS Cut Line= 4
 2157418.4337122656795.3413467212157217.59048321656991.585890366
2156856.93019322657059.3058717422156664.92383575657100.726246048
#Sta/Elev= 30
       0 1609.46    14.3 1606.99    64.7 1588.74    84.9 1590.18    99.9 1584.41
   117.1 1583.02     140 1573.59   154.2 1569.96   186.8 1568.23   210.1 1564.22
   226.9 1558.66   243.6 1550.39   300.6 1531.22   343.3 1520.63   365.8  1509.7
  381.511495.414   389.6 1491.47   404.3 1490.83   428.8 1491.04   444.11495.418
   461.3 1501.03   542.7 1500.84   611.9 1504.97   636.3 1510.81   673.1 1509.02
   689.5 1517.43   808.1 1548.37   824.5 1551.92   836.8 1552.36   844.2 1556.05
#Mann= 8 ,-1,0
       0      .1       0   380.8     .05       0  381.51    .045       0
   444.1     .05       0   480.8     .06       0   580.8      .1       0
  677.77     .08       0  787.77      .1       0
Bank Sta=381.51,444.1
XS Rating Curve= 0 ,0
Exp/Cntr=0.3,0.1

Type RM Length L Ch R = 1 ,32712   ,418,437.4,429
XS GIS Cut Line= 3
2156832.55536817656336.5285054662156616.36239649656674.972653611
     2156522.124 656812.74810674
#Sta/Elev= 30
       0 1586.67    19.8 1576.16    29.7 1569.11      34 1567.51    45.3 1565.86
    57.7  1560.4    86.2 1542.22    95.7 1536.92   109.9 1531.95   147.9 1511.15
  183.361495.125   193.9 1491.44   200.1 1490.81     244 1490.31   252.3 1491.33
  263.031495.127   270.1 1496.08   283.1 1496.02   295.1 1498.15   309.3 1497.57
   318.8 1499.92   345.4 1501.86     357 1504.15     371 1505.43   380.5 1508.38
   385.2 1509.02   418.8 1508.49   447.9 1521.61   496.4 1534.17   568.5 1554.17
#Mann= 6 ,-1,0
       0      .1       0  183.36    .045       0  263.03     .06       0
     380      .1       0   501.6     .08       0   551.6      .1       0
Bank Sta=183.36,263.03
XS Rating Curve= 0 ,0
Exp/Cntr=0.3,0.1

Type RM Length L Ch R = 1 ,32275   ,383,396.6,387.2
XS GIS Cut Line= 3
2156502.45686055656105.5045751922156278.99109366656452.489631833
2156194.01602832656615.700479298
#Sta/Elev= 30
       0 1583.36    61.5  1552.7    66.2 1550.91      71 1550.15    75.7 1548.23
     109  1526.9     152 1504.61   166.7  1499.1   188.61494.097   212.7 1490.68
   215.6 1490.86  228.561494.097   242.3 1497.99   267.7 1500.92   289.8 1501.82
   308.2  1501.2   318.4  1499.9   331.3 1499.98   348.7 1501.14   357.4 1504.24
   361.2 1504.87     418 1504.22     427  1507.7   468.7 1514.88   476.6 1516.88
   486.5 1518.17   512.7 1528.23   530.7  1533.5   551.7 1538.78   596.7  1548.4
#Mann= 5 ,-1,0
       0      .1       0   188.6    .045       0  228.56      .1       0
     310     .06       0  422.72      .1       0
Bank Sta=188.6,228.56
XS Rating Curve= 0 ,0
Exp/Cntr=0.3,0.1

Type RM Length L Ch R = 1 ,31878   ,427.4,422.2,402.5
XS GIS Cut Line= 3
2156158.13554902655932.8254967722155980.40730937 656239.75700439
2155920.85452724656427.497021778
#Sta/Elev= 30
       0 1573.83    32.8 1559.37    45.6 1552.97     116 1520.64   139.3 1508.96
   152.9 1497.84   157.6 1494.86  164.221492.419   180.7 1489.86   189.9 1489.29
   203.8 1490.37   226.9 1489.77   231.5 1490.38  235.861492.422   245.4 1495.74
   254.6 1496.85   263.9 1500.11   267.3 1500.41   309.1 1501.21   347.1 1503.47
     391 1504.19   413.3  1502.4   435.9 1502.04   440.1    1503     448 1509.09
   451.6 1511.17   456.9 1512.67   502.5 1518.48   540.7 1520.15   551.6 1521.97
#Mann= 6 ,-1,0
       0      .1       0  164.22    .045       0  235.86      .1       0
     270     .07       0  384.67     .06       0  484.67      .1       0
Bank Sta=164.22,235.86
XS Rating Curve= 0 ,0
Exp/Cntr=0.3,0.1

Type RM Length L Ch R = 1 ,31456   ,313,281.1,221
XS GIS Cut Line= 3
2155701.27904509655791.6191274862155680.00702157656062.333800017
2155753.75408823656421.335847052
#Sta/Elev= 30
       0 1559.49     9.6 1557.15    25.6 1550.58    49.7  1543.9    65.8 1536.78
    85.8 1525.15    93.8 1518.84   105.9 1512.14   118.1 1506.91     138 1492.94
  145.321489.624   151.3 1488.13   170.1 1487.62  199.321489.625   202.2 1490.51
   210.2 1495.93   218.2 1497.28   282.6 1498.87   364.3 1499.07     401 1501.22
   462.3  1501.6   503.1 1507.53   523.5 1512.81     544    1517   584.8 1519.08
   601.1 1519.15   605.2 1520.06   617.5 1525.07   625.6 1526.65     638 1530.93
#Mann= 7 ,-1,0
       0      .1       0  145.32    .045       0  199.32      .1       0
  281.55     .08       0  381.55     .06       0  481.55     .05       0
  581.55      .1       0
Bank Sta=145.32,199.32
XS Rating Curve= 0 ,0
Exp/Cntr=0.3,0.1

Type RM Length L Ch R = 1 ,31175   ,82,78.2,78.2
XS GIS Cut Line= 4
2155420.02428189655897.5878111032155426.39186814 656044.22613654
2155686.38185736656158.624711803 2155729.5421106656424.598927034
#Sta/Elev= 30
       0 1533.47    19.6  1527.6    31.6 1518.37    39.6 1513.88    71.7  1504.3
   143.7 1500.55     169 1497.43   179.3 1497.22   188.1 1495.03  200.791488.487
   209.9  1485.9   238.5 1486.66   261.1  1485.6  301.261488.488   327.9 1496.47
     341 1498.29   385.6 1499.63   430.8 1499.47   460.8 1501.43   490.1 1500.19
   530.7 1502.02     559 1506.28   603.6 1516.81   626.4 1517.68   644.1 1519.71
   656.3 1519.01   664.4  1519.7   671.7 1521.88   692.6 1531.52   700.3 1533.12
#Mann= 9 ,-1,0
       0     .06       0      70     .07       0  196.78      .1       0
  200.79    .045       0  301.26     .07       0  396.78     .08       0
  440.82     .06       0  540.82     .05       0  640.82      .1       0
Bank Sta=200.79,301.26
XS Rating Curve= 0 ,0
Exp/Cntr=0.3,0.1

Type RM Length L Ch R = 1 ,31097   ,73.5,98,133.1
XS GIS Cut Line= 4
2155371.15769266655927.7752908272155380.44304968656107.967980291
2155640.43303891656222.3665555552155671.92220901656421.232042729
#Sta/Elev= 30
       0 1525.63    21.4 1519.54    41.5 1511.36    65.5 1508.27    86.1 1503.87
   105.5 1501.62   145.6 1501.39   161.6 1499.54   254.4  1499.2   258.8 1498.78
   263.2 1497.18   271.9 1491.74  279.261488.377     285 1486.28   289.4 1485.61
   302.4 1485.25   351.1 1485.74   365.11488.376   375.4 1489.61   384.5 1491.75
   394.3 1496.17   398.6 1497.24   423.9 1499.33   461.5 1499.23   479.5 1500.76
   495.7 1503.79   544.3 1507.65   596.9 1517.23   641.9 1527.34   665.8 1533.63
#Mann= 7 ,-1,0
       0     .06       0      40     .07       0     140      .1       0
  279.26    .045       0   365.1     .06       0  514.48     .05       0
  604.48      .1       0
Bank Sta=279.26,365.1
XS Rating Curve= 0 ,0
Exp/Cntr=0.3,0.1

Type RM Length L Ch R = 1 ,30999   ,193.7,209.8,233.8
XS GIS Cut Line= 4
2155302.39321223655932.7935182792155342.85467672656122.327496277
2155395.41414704656140.844498618 2155509.6050749656444.386823271
#Sta/Elev= 30
       0 1529.03    12.7 1523.55    24.9 1516.85    69.9 1511.36    82.2 1501.99
    86.3  1500.9   110.8 1501.67   155.8 1499.68   193.8 1495.22   212.2  1495.9
   237.6 1498.81   249.9 1498.77   258.4 1497.83   279.8 1492.91   296.9 1491.38
   308.5 1488.44     314 1485.71   322.5 1485.14     361 1486.27   365.3 1486.69
   367.81488.321   369.6  1489.5   374.6 1495.41   378.1 1498.01   380.8 1498.66
   412.3 1499.61   463.6 1506.56   484.9 1511.88   519.1 1513.75   573.8 1530.93
#Mann= 7 ,-1,0
       0     .06       0      40      .1       0  279.53     .06       0
   308.5    .045       0   367.8     .06       0  409.53     .05       0
  489.53      .1       0
#XS Ineff= 2 , 0
          244.54 1501.08
Permanent Ineff=
       F       F
Bank Sta=308.5,367.8
XS Rating Curve= 0 ,0
Exp/Cntr=0.3,0.1

Type RM Length L Ch R = 1 ,30789   ,204,250.1,245
XS GIS Cut Line= 4
2155279.10349998655927.0040984852155259.67123651656146.200030431
2155193.60154071 656296.994394962155206.81547987656445.456887874
#Sta/Elev= 30
       0  1533.7     6.2 1530.44    18.2  1521.6    23.1  1520.6    42.3 1520.06
      49 1518.16    54.4 1514.68    66.4 1503.15    70.5 1501.67   106.6 1501.82
   130.7 1495.97   150.8 1494.09     267  1491.6   289.71486.115   300.9 1484.01
   319.4 1484.67   328.1 1483.85   337.3 1484.36  343.251486.208   348.4 1488.15
   358.7 1488.33   374.5 1499.36   378.3  1500.8     405 1500.48   433.1 1502.29
   453.1 1506.59   474.6 1509.21   497.3 1510.58   513.4 1515.94   533.7 1520.15
#Mann= 6 ,-1,0
       0     .06       0      40      .1       0   289.7    .045       0
  343.25      .1       0  350.06     .06       0  454.69      .1       0
#XS Ineff= 2 , 0
          261.06 1499.16
Permanent Ineff=
       F       F
Bank Sta=289.7,343.25
XS Rating Curve= 0 ,0
Exp/Cntr(USF)=0,0
Exp/Cntr=0.3,0.1

Type RM Length L Ch R = 1 ,30539   ,246.1,223.4,205
XS GIS Cut Line= 4
2155215.56729104655897.7931026462155151.56916279656052.570893038
2155000.85435262656133.8076576942154924.25495032656378.758363868
#Sta/Elev= 30
       0 1535.44     8.3 1531.68    23.6 1530.58    29.6 1529.32    48.1 1521.44
    55.6 1517.17    64.3 1506.99    69.5 1503.48    72.9 1502.92    94.6 1503.66
   103.1 1503.08   111.9 1501.68   120.5 1497.93   133.8 1494.72   155.2 1491.82
     185 1489.87   194.1  1488.5   207.7 1482.56   216.8 1480.88   236.2 1481.54
   253.1 1480.22   284.9 1480.81     294 1482.61   300.4 1483.48   312.2 1486.69
   330.4  1494.1   354.7 1495.13   364.3 1498.04   522.4 1509.38   595.3 1516.53
#Mann= 6 ,-1,0
       0     .06       0      80      .1       0     160     .06       0
   207.7    .045       0     294     .05       0   368.7      .1       0
Bank Sta=207.7,294
XS Rating Curve= 0 ,0
Exp/Cntr(USF)=0,0
Exp/Cntr=0.3,0.1

Type RM Length L Ch R = 1 ,30315   ,264,259.7,254.9
XS GIS Cut Line= 3
2155009.96132155655762.7691510032154894.30455097655999.624274511
2154661.13199019656237.760749006
#Sta/Elev= 30
       0  1567.5     2.7 1566.98    20.5 1554.72    38.3 1553.48    51.6 1545.18
    65.9  1541.6    69.5 1538.73    80.9 1520.33    86.9 1513.13    91.7    1509
    96.2  1507.5   122.9 1508.32   128.8 1507.18   140.7 1498.81     154  1484.5
  159.971479.624   176.3 1477.92  222.741479.623   233.4 1481.12   248.4 1488.38
   260.4 1489.94   325.6 1492.12   362.4 1496.17   398.1  1497.2   426.7 1495.53
   478.3 1499.85   512.1 1507.79   563.2 1514.59   575.4 1519.35   596.9 1523.18
#Mann= 8 ,-1,0
       0      .1       0      10     .06       0     120     .07       0
  159.97    .045       0  222.74     .07       0     230     .06       0
  313.58     .05       0  353.58      .1       0
Bank Sta=159.97,222.74
XS Rating Curve= 0 ,0
Exp/Cntr=0.3,0.1

Type RM Length L Ch R = 1 ,30056   ,307.9,316.2,320.1
XS GIS Cut Line= 4
2154770.34346254655664.5735295212154709.11226955655760.529143543
2154673.38617933655932.8697812592154541.02127688656128.976262709
#Sta/Elev= 30
       0 1551.18     4.9 1547.59    16.5 1541.32    19.4 1538.06    24.4  1530.2
    28.1 1526.56      31 1525.87    57.7 1526.08    62.8 1524.95    71.9 1519.09
    95.6 1499.07   118.6 1482.83     139 1473.57   159.8 1469.33   204.4 1467.25
  214.16  1465.5   224.8 1462.58   228.9 1462.21     237 1463.43   242.81465.502
   249.3 1468.05   273.8 1483.29   277.9 1484.68   328.4 1485.87     342 1488.85
     435 1496.25   449.5 1499.26   478.4 1506.92   512.2 1508.08   526.4 1512.35
#Mann= 6 ,-1,0
       0     .06       0      20      .1       0  123.83     .06       0
  214.16    .045       0   242.8     .06       0  449.83      .1       0
Bank Sta=214.16,242.8
XS Rating Curve= 0 ,0
Exp/Cntr=0.3,0.1

Type RM Length L Ch R = 1 ,29739   ,424.3,421.1,402.4
XS GIS Cut Line= 3
2154609.26148774655508.9376884742154403.36433459655721.742552257
2154380.74718799656026.817177384
#Sta/Elev= 30
       0 1552.75    13.1  1545.3    44.9  1545.6    54.7 1542.47    87.9 1516.88
   106.1 1508.11   116.6 1500.78   122.4 1492.54   128.2 1479.97   131.1 1476.29
  150.131459.541   156.2 1457.63   168.4 1457.33  193.071459.545   266.2  1466.8
   317.2 1469.04   331.6 1472.39   351.7 1480.56   383.8  1473.9   415.9 1475.21
   436.7 1473.33     468 1476.35     480  1475.8   496.1 1483.25   520.2 1484.75
   532.2 1495.37   544.2 1502.41   571.2 1513.11   588.3  1523.9     602 1526.18
#Mann= 3 ,-1,0
       0      .1       0  150.13    .045       0  193.07      .1       0
Bank Sta=150.13,193.07
XS Rating Curve= 0 ,0
Exp/Cntr=0.3,0.1

Type RM Length L Ch R = 1 ,29318   ,416.3,438.9,425.4
XS GIS Cut Line= 3
2154193.06813846655286.0465783382154099.10308181 655612.79382693
2153978.37996539655836.619166777
#Sta/Elev= 30
       0 1523.91    25.9 1522.12    32.4 1519.83    40.7 1513.11    44.9 1511.18
    57.4 1508.05    69.9 1507.04    78.2  1503.1    94.8 1489.21   104.5 1471.93
   116.4 1464.14   161.6 1456.74     203 1454.55   215.5 1455.12  238.191450.593
   269.6 1448.38  281.211450.595   290.9 1456.58   340.4 1473.57   358.6 1472.66
   372.2 1469.77   422.2 1469.34   451.7 1471.81   475.3 1476.25   508.6 1477.05
   513.7 1478.65   531.5 1492.31   572.7 1516.95   581.3 1520.72   594.3 1523.34
#Mann= 5 ,-1,0
       0      .1       0  238.19    .045       0  281.21      .1       0
     300     .06       0  409.99      .1       0
Bank Sta=238.19,281.21
XS Rating Curve= 0 ,0
Exp/Cntr=0.3,0.1

Type RM Length L Ch R = 1 ,28879   ,341.7,344.7,341.3
XS GIS Cut Line= 3
2153893.77168599655115.8098898642153760.90535558655363.736034614
2153602.80103147655641.165122722
#Sta/Elev= 30
       0  1528.1    19.7 1520.65    61.3 1507.49    65.1 1505.61    74.2 1497.62
    92.3 1496.39   105.6 1486.25   129.2 1465.15   141.1 1456.74   151.3 1447.77
  171.511440.605   201.2  1439.7     212 1438.14   243.11440.606   253.3 1443.01
   260.2 1445.92   273.8 1448.31   292.2 1449.38   306.3 1447.14   323.2 1447.58
     375 1455.38   425.7 1455.94   444.2 1454.97     497  1457.9   500.9 1459.39
   508.5 1468.41   513.1 1472.42     527 1476.73   555.6 1492.64   600.6 1503.27
#Mann= 5 ,-1,0
       0      .1       0  171.51    .045       0   243.1      .1       0
  301.28     .06       0  451.28      .1       0
Bank Sta=171.51,243.1
XS Rating Curve= 0 ,0
Exp/Cntr=0.3,0.1

Type RM Length L Ch R = 1 ,28535   ,212.4,228.7,236.1
XS GIS Cut Line= 3
2153683.42549895655054.7630909982153503.00322942655144.888378313
2153298.68314169655503.871498222
#Sta/Elev= 30
       0 1475.24    21.5 1465.61    39.4 1461.94    48.3 1458.64    66.2 1454.38
      77 1449.31   124.4 1445.71   132.4 1443.43   147.4 1441.54   195.9 1439.62
   220.4 1440.45   224.5 1439.36   233.3 1434.31     245  1431.9   261.8 1431.55
   288.3 1432.35  299.451434.292   340.1 1444.15   399.9  1442.4   445.9 1445.08
   458.1 1447.12   482.8 1448.04   501.2 1454.57   528.8 1468.67   542.6 1473.58
     561 1477.18   579.4  1477.5     584 1478.56   600.8 1487.81   614.7 1492.65
#Mann= 3 ,-1,0
       0      .1       0   233.3    .045       0  299.45      .1       0
Bank Sta=233.3,299.45
XS Rating Curve= 0 ,0
Exp/Cntr=0.3,0.1

Type RM Length L Ch R = 1 ,28306   ,218.7,262.9,287.2
XS GIS Cut Line= 4
2153625.98147201 654920.662817492153367.22839742 655010.86602061
2153264.68734614655083.2950755212153079.09313846655110.326726894
#Sta/Elev= 30
       0 1474.46    48.5  1459.3    69.7 1458.42    82.4 1455.61   107.8 1448.39
     129  1439.6   136.9 1437.97   167.1  1436.8   188.3 1433.93   209.5 1435.23
   234.9 1433.94   268.7 1435.22   287.6 1435.09   292.5 1433.42   297.4 1429.75
  303.051427.824   321.8    1426     341 1425.68  365.721427.825   370.8  1429.4
   385.5 1440.78   395.5 1446.88   404.1 1449.54   412.2 1453.64   452.6 1458.18
   464.8 1462.02   489.9 1466.59   505.2 1470.76   533.5 1474.37   587.1  1486.9
#Mann= 3 ,-1,0
       0      .1       0  303.05    .045       0  365.72      .1       0
Bank Sta=303.05,365.72
XS Rating Curve= 0 ,0
Exp/Cntr=0.3,0.1

Type RM Length L Ch R = 1 ,28043   ,421.9,396.9,357.5
XS GIS Cut Line= 4
2153616.05188799654815.1249892852153422.34058742654842.631516156
2153294.47570869654782.1356372392153048.40674197654823.783773436
#Sta/Elev= 30
       0 1475.86    40.3 1464.28    48.4 1460.96    65.4 1459.59     117 1450.18
   125.1 1445.96   133.2 1443.28   145.3 1436.83   165.5 1435.18   189.8 1435.19
   202.5 1432.08   215.8 1425.35 232.4141422.934   270.5 1421.12   297.5 1421.44
   308.7    1423   337.1 1429.81   351.6 1430.84   367.8 1436.29   396.2  1441.1
   420.6 1447.18     449 1450.55   461.1 1453.65   472.9 1453.47   485.5 1454.82
   509.8 1461.05   531.5 1469.92   550.4 1473.53   566.6  1481.2   586.7 1481.94
#Mann= 3 ,-1,0
       0      .1       0 232.414    .045       0   308.7      .1       0
Bank Sta=232.414,308.7
XS Rating Curve= 0 ,0
Exp/Cntr=0.3,0.1

Type RM Length L Ch R = 1 ,27646   ,302.5,309.2,311
XS GIS Cut Line= 4
2153518.96426348654389.8469517112153361.26716325654419.714712084
2153160.02874932654515.5897904822152986.86972539 654563.63637652
#Sta/Elev= 30
       0 1466.12    19.1 1459.28      72 1447.11   100.5 1442.75   118.2 1441.17
   141.3  1440.1   161.7  1440.3   170.6 1439.09   192.4 1431.61   197.2 1428.36
   207.4 1418.41  213.26 1414.63     229 1413.72   264.5 1414.64   294.6  1414.3
     312 1421.03   321.2    1422   334.5 1426.38   356.7 1437.47   365.5 1439.99
   383.2    1442   391.6 1446.21   424.8 1446.92   437.2 1452.11   466.3 1460.37
   495.1 1470.86   507.8 1476.62   520.2 1480.73   547.5 1494.24   563.1 1500.23
#Mann= 3 ,-1,0
       0      .1       0  213.26    .045       0   264.5      .1       0
Bank Sta=213.26,264.5
XS Rating Curve= 0 ,0
Exp/Cntr=0.3,0.1

Type RM Length L Ch R = 1 ,27337   ,339.6,339.7,328.5
XS GIS Cut Line= 3
2153450.09569932      654131.626 2153113.8705294654191.160662305
2152960.84456865 654272.92059258
#Sta/Elev= 30
       0  1452.1    54.8 1447.56    87.3 1447.91   123.8 1445.87   131.9 1446.32
     136 1445.48     141 1443.07   164.4  1428.9   180.7 1420.73   192.9 1418.74
   205.1 1415.13   217.2 1409.06   229.4 1408.11   241.6 1410.94  251.221408.869
   261.9 1406.66  294.171408.886   306.7 1412.05   322.9  1428.8   326.9 1430.78
   339.1 1432.76   347.9 1436.31   352.4 1436.93   382.6 1436.51   393.3 1438.83
   443.2 1445.08   470.4 1454.47   479.4  1456.3   498.5 1463.84     515 1468.68
#Mann= 3 ,-1,0
       0      .1       0  251.22    .045       0  294.17      .1       0
Bank Sta=251.22,294.17
XS Rating Curve= 0 ,0
Exp/Cntr=0.3,0.1

Type RM Length L Ch R = 1 ,26997   ,356.1,354.7,331.4
XS GIS Cut Line= 4
2153316.50615878653736.1863411732153239.36165266653832.322344172
2153094.31224313653879.3377784452152836.88192158654096.591701971
#Sta/Elev= 30
       0 1474.31    13.3 1469.29    26.6 1468.64    40.8 1463.87    47.4 1460.77
    96.4 1448.69   103.4 1445.43   119.2 1435.94   145.6 1417.11   161.4  1404.5
  172.081399.565   185.5  1397.7   206.5 1397.59   219.1 1398.34   224.51399.568
   240.1 1404.13   273.8 1408.22   320.4 1405.75   363.7 1408.07   383.2 1406.46
   406.3 1406.21     446  1420.4   457.4 1423.32   472.2 1430.71   493.1 1431.31
   502.8 1435.64   529.8 1441.95   568.1 1453.38   592.6 1462.66   612.6 1471.29
#Mann= 3 ,-1,0
       0      .1       0  172.08    .045       0   224.5      .1       0
Bank Sta=172.08,224.5
XS Rating Curve= 0 ,0
Exp/Cntr=0.3,0.1

Type RM Length L Ch R = 1 ,26643   ,392.8,390.8,379.7
XS GIS Cut Line= 3
 2153056.5788301653507.954818826  2152969.046496653689.757897477
2152738.80343089653928.297138229
#Sta/Elev= 30
       0 1444.47    40.2 1413.47    58.2 1394.79   60.251393.402      68 1391.48
    81.3 1393.34   103.5 1392.36   112.1  1394.1   121.2 1397.48   130.1 1398.85
   134.5 1398.56   143.4 1394.96   147.9 1394.53   161.2 1396.97   187.8 1398.48
   201.1  1401.2   237.6 1397.09   255.7 1399.93   295.3 1399.34   362.2 1403.02
   387.3 1400.13   408.5 1401.76   417.8 1404.67   428.9 1410.34   451.1 1426.03
   456.5 1428.68     468 1429.08   479.2 1434.43   506.7 1440.17   533.3 1447.93
#Mann= 3 ,-1,0
       0      .1       0   60.25    .045       0    81.3      .1       0
#XS Ineff= 2 , 0
                           260.1         1404.11
Permanent Ineff=
       F       F
Bank Sta=60.25,81.3
XS Rating Curve= 0 ,0
Exp/Cntr=0.3,0.1

Type RM Length L Ch R = 1 ,26252   ,298.2,306.3,320.6
XS GIS Cut Line= 4
2152693.88999346653435.3162353452152646.25502148653505.845925682
2152652.67992158653691.2942374972152558.84585186653829.765466213
#Sta/Elev= 30
       0 1438.89     7.1 1438.39    10.2 1436.97    19.9  1430.7    38.8 1420.79
    50.5 1411.08    57.3 1407.31    71.7 1403.57    92.4 1401.55    96.4 1399.76
   104.5 1390.92  109.86 1386.98   116.5 1385.33   136.5  1386.9   176.5 1385.97
   188.5 1387.95   196.5 1387.89   232.5 1394.09   260.5 1395.21   271.6 1396.89
   277.8 1398.84   286.8 1403.54   311.6 1421.75   321.4 1427.21   350.3 1428.32
   364.8 1431.22   395.8 1434.76   427.6  1443.1   432.4 1446.55   437.9 1451.83
#Mann= 3 ,-1,0
       0      .1       0  109.86    .045       0   136.5      .1       0
Bank Sta=109.86,136.5
XS Rating Curve= 0 ,0
Exp/Cntr=0.3,0.1

Type RM Length L Ch R = 1 ,25946   ,297,301.8,272.7
XS GIS Cut Line= 3
2152548.52537471653244.1092723592152309.92953594653508.012723336
2152266.36881484653627.782838771
#Sta/Elev= 30
       0  1444.3      23 1436.95    66.2 1425.09      96 1419.86   120.1  1418.4
   130.9 1413.38   143.7 1404.02   176.6 1382.87  182.031380.454   196.4 1378.48
   215.2 1379.83   233.1 1378.65  241.141380.457   255.9 1387.03   264.4 1388.42
   271.1 1390.87   298.4 1405.42   306.9 1410.89   314.2 1413.66     325 1414.38
   343.7 1419.73   369.8 1421.27   379.9 1423.82     396 1422.05   411.1 1424.02
   425.1 1429.19   433.6 1425.52   437.9 1425.35   463.4 1432.57   483.2  1435.8
#Mann= 3 ,-1,0
       0      .1       0  182.03    .045       0  241.14      .1       0
Bank Sta=182.03,241.14
XS Rating Curve= 0 ,0
Exp/Cntr=0.3,0.1

Type RM Length L Ch R = 1 ,25644   ,363.3,349,297.7
XS GIS Cut Line= 3
2152319.07429414653067.9051350612152105.03771856653392.402997559
 2152077.6129499653528.002409572
#Sta/Elev= 30
       0 1442.86    30.3 1436.86    43.4 1430.97    63.4  1418.8    73.4 1410.32
    92.4 1397.19     107 1389.66   118.5 1381.39   126.1 1377.04   132.81374.503
   158.9 1372.79   190.7 1373.09  202.261374.503   216.7 1375.27   231.5 1380.16
   237.7 1380.99   277.3  1381.7   303.3 1381.09   317.8 1384.92   332.2 1393.56
   346.5 1404.57   351.3 1406.09   375.3 1407.69   384.1 1409.29   393.5 1406.77
   397.7 1406.83   426.2 1410.14   458.9 1411.79   487.5 1416.14   527.1 1428.88
#Mann= 3 ,-1,0
       0      .1       0   132.8    .045       0  202.26      .1       0
Bank Sta=132.8,202.26
XS Rating Curve= 0 ,0
Exp/Cntr=0.3,0.1
