HEC-RAS study LIKANARV.prj: LIKANARV

--- LIKANARV.g01 (geometry) --- (continued)

Type RM Length L Ch R = 1 ,25295   ,352.8,390.3,400.1
XS GIS Cut Line= 3
2151871.20003486653028.6052571232151970.88237256653266.874076267
2151928.14442266653504.239649221
#Sta/Elev= 30
       0 1411.82    48.3 1405.52    52.7 1403.53    64.7 1393.91    75.1 1387.64
    87.3 1381.03      96 1378.13   113.4 1366.84  118.89 1365.78   161.1  1363.8
   183.61365.779   195.7 1369.13   208.7 1374.21   224.3 1375.02   247.8 1374.28
     258 1376.64   289.1 1387.98     297 1397.02   301.3 1398.98   307.3 1399.63
   325.7 1399.44     346 1403.86   354.1 1402.25   358.2 1402.24   370.4  1403.6
   393.5 1403.17     411 1405.02   456.1 1413.98   484.2 1422.78   499.5 1428.35
#Mann= 5 ,-1,0
       0      .1       0  118.89    .045       0   183.6      .1       0
     200     .06       0  308.28      .1       0
Bank Sta=118.89,183.6
XS Rating Curve= 0 ,0
Exp/Cntr=0.3,0.1

Type RM Length L Ch R = 1 ,24904   ,368.4,374.8,377.5
XS GIS Cut Line= 4
2151775.91028105653003.4078627872151622.15695644653091.367359473
2151534.27798644653230.5104855512151498.98663838653348.319769045
#Sta/Elev= 30
       0 1409.66      89 1400.32   150.6 1392.19   172.7 1388.01   182.8 1385.31
   188.7 1382.63   198.2 1376.88   212.4 1366.89  231.281355.357   237.9 1352.96
   250.2 1352.63   261.1  1353.3  266.351355.356   272.7 1359.23   283.4 1362.49
   302.3 1363.66   307.5 1364.42   311.7 1365.73   330.7 1381.57   335.4 1383.19
   340.1 1383.38   344.5 1384.55   352.8 1391.09   361.6 1394.96   373.7 1395.81
   386.2 1398.47   398.8 1399.03   407.1  1400.1   454.8  1410.4   464.7 1413.17
#Mann= 3 ,-1,0
       0      .1       0  231.28    .045       0  266.35      .1       0
Bank Sta=231.28,266.35
XS Rating Curve= 0 ,0
Exp/Cntr=0.3,0.1

Type RM Length L Ch R = 1 ,24530   ,342.2,341.6,320
XS GIS Cut Line= 3
2151413.83089541652805.4145316352151231.29224619652985.689483688
2151204.73118086653132.440015236
#Sta/Elev= 30
       0 1392.78    34.9 1380.96    43.4  1379.4    49.1 1376.33    58.5 1369.26
    79.4 1357.28    94.3 1351.77   103.5 1349.01  108.281348.163   120.4 1347.41
   142.4 1347.83   153.4 1347.23   167.9 1348.19     182 1347.54   207.5 1349.25
   221.7 1352.26   227.4 1353.93   244.4 1361.58   249.7 1362.69   255.8 1362.99
   268.2 1368.96   272.3 1370.49   280.4 1372.88   288.6 1374.69   304.8 1377.72
   329.2 1381.07   355.2 1385.45   369.9 1386.35   386.4 1388.82   405.7 1392.84
#Mann= 3 ,-1,0
       0      .1       0  108.28    .045       0   167.9      .1       0
Bank Sta=108.28,167.9
XS Rating Curve= 0 ,0
Exp/Cntr=0.3,0.1

Type RM Length L Ch R = 1 ,24188   ,348.1,359.7,338.6
XS GIS Cut Line= 3
2151105.19176035652584.5661721612151050.44643574652745.967069726
2150984.02985185 653030.87118516
#Sta/Elev= 30
       0 1394.28     9.1 1393.81    13.3 1392.01    76.7 1344.67    83.3 1342.66
    89.6 1341.42   106.2  1341.2  132.751342.683   148.5 1346.33   165.3 1348.05
   190.2 1346.14   198.4  1347.8   231.2 1348.14   251.8 1343.54   264.9 1337.85
   276.4 1336.62   284.6 1336.94   292.8 1339.06   309.3 1347.58   317.5 1347.66
   321.6 1349.11   325.7 1352.63   329.8 1354.82   348.2 1357.13   362.7 1361.68
   379.1  1361.9   391.5 1364.38   407.8 1369.55   436.6 1372.57     463  1384.1
#Mann= 3 ,-1,0
       0      .1       0    83.3    .045       0  132.75      .1       0
Bank Sta=83.3,132.75
XS Rating Curve= 0 ,0
Exp/Cntr=0.3,0.1

Type RM Length L Ch R = 1 ,23828   ,290.9,331.5,341.3
XS GIS Cut Line= 3
 2150942.6795843652582.3979608332150800.77506472652719.176166652
2150766.93734904652945.626235259
#Sta/Elev= 30
       0 1364.26     9.8 1362.31    20.1 1361.06    36.8 1360.33      49 1358.26
    63.1 1358.43   105.6 1353.63   125.4 1353.06   136.6    1350   142.4 1349.16
     148 1348.99     159  1350.3   176.3 1349.35   194.2 1350.26   219.3 1345.63
   235.5 1341.24   247.6 1337.24   259.8 1335.71  270.46 1331.75     284  1330.1
   316.4 1330.32  326.421331.751   332.6 1332.72   336.7 1334.87   344.7 1342.71
   352.8 1348.07   360.9 1354.51   389.2  1375.1   393.2 1377.37   426.1 1387.29
#Mann= 3 ,-1,0
       0      .1       0  270.46    .045       0  326.42      .1       0
Bank Sta=270.46,326.42
XS Rating Curve= 0 ,0
Exp/Cntr=0.3,0.1

Type RM Length L Ch R = 1 ,23497   ,283.7,335.1,333.9
XS GIS Cut Line= 5
2150794.26964115652435.9489078762150696.24642551652556.056045089
2150588.21123379652609.1741146472150478.66790632652683.621036227
2150457.19243533652771.780276457
#Sta/Elev= 30
       0  1364.8    33.6 1352.96    42.2 1349.25    56.4  1347.9    73.9 1343.88
    84.8 1340.34   110.9 1339.06   167.9 1338.26   177.4 1334.81   190.8 1327.61
   199.7  1326.6   213.1 1326.62   245.6 1329.82   262.1 1330.17     271 1331.63
   284.1 1330.97     290 1330.23  303.221324.085   309.3 1322.86   323.8  1322.5
   357.7 1322.78  370.751324.084   384.9 1328.64   407.9 1340.18   413.6 1342.16
   425.9 1349.14   438.3 1352.36   447.6 1356.53   480.7 1378.34   498.6 1386.45
#Mann= 3 ,-1,0
       0      .1       0  303.22    .045       0  370.75      .1       0
#XS Ineff= 2 , 0
          266.71 1338.33
Permanent Ineff=
       F       F
Bank Sta=303.22,370.75
XS Rating Curve= 0 ,0
Exp/Cntr=0.3,0.1

Type RM Length L Ch R = 1 ,23162   ,434.6,414.6,381.9
XS GIS Cut Line= 5
2150750.42040698652349.2139103212150675.79750266652389.524670159
 2150539.4652292652386.3088768952150414.41679581652346.583278653
2150235.03136885652443.096646262
#Sta/Elev= 30
       0 1358.82     8.3 1354.29    25.2 1346.94    52.6 1338.23    75.7 1333.33
    88.4 1328.38   104.3 1325.04   180.5 1320.83   192.5 1321.73   200.5 1323.37
   220.5 1324.15   245.6 1321.64260.72731316.248   270.8 1314.47   287.6 1313.91
   317.1 1314.41   323.4 1316.31   330.6 1321.48   342.2 1328.06   350.5 1330.34
     364 1337.34   368.6 1338.33   382.2 1339.03   423.1 1338.12   441.2 1339.12
   468.5 1339.02   486.7 1340.71   500.3 1344.41   541.2 1349.36   556.1 1352.63
#Mann= 3 ,-1,0
       0      .1       0260.7273    .045       0   323.4      .1       0
Bank Sta=260.7273,323.4
XS Rating Curve= 0 ,0
Exp/Cntr=0.3,0.1

Type RM Length L Ch R = 1 ,22747   ,366.1,344.1,316.2
XS GIS Cut Line= 3
2150637.19805879 651904.307601982150445.08242941 652030.61488825
2150137.54258041652269.239605871
#Sta/Elev= 30
       0 1432.72       6 1430.18    25.2 1418.01    30.2 1413.81    34.7 1406.73
    44.3 1384.58    50.5  1376.1    58.7 1360.91      62 1356.78    74.4 1347.46
    90.9  1329.6   108.2 1312.95  118.721307.159   125.6 1305.38   144.8 1305.23
  179.091307.158   197.5 1313.05   216.6 1315.47   235.2 1315.49   266.6 1313.15
   289.4 1314.15   299.4 1315.73   312.4 1315.22   332.3  1319.5   358.1 1322.02
   398.1 1328.44   442.9  1327.9   462.5 1325.86   534.8 1326.89   619.2 1341.83
#Mann= 3 ,-1,0
       0      .1       0  118.72    .045       0  179.09      .1       0
Bank Sta=118.72,179.09
XS Rating Curve= 0 ,0
Exp/Cntr=0.3,0.1

Type RM Length L Ch R = 1 ,22403   ,348.7,368.9,380
XS GIS Cut Line= 3
 2150252.8262374651713.154354615 2150238.8833813652087.811493042
2150123.54544082652237.685659978
#Sta/Elev= 30
       0 1353.59      20 1347.43      28 1343.53    48.1 1323.64    65.9 1307.91
    68.1 1306.06    76.1 1302.85    80.1 1302.39   116.1 1304.82   124.1 1303.71
   136.1 1300.51   160.1 1300.38   184.2 1298.58  196.681300.405   220.2 1308.92
   224.2 1308.99   236.3 1306.58   248.2 1305.63   268.2 1308.44   312.2 1309.38
   324.2 1312.19   351.8 1321.64   368.3 1325.48   379.4 1326.03   406.9 1323.92
   464.6  1324.9   490.9 1329.42     504 1329.35   536.8 1332.21     564 1338.42
#Mann= 3 ,-1,0
       0      .1       0   160.1    .045       0  196.68      .1       0
#XS Ineff= 2 , 0
                          220.42         1314.33
Permanent Ineff=
       F       F
Bank Sta=160.1,196.68
XS Rating Curve= 0 ,0
Exp/Cntr=0.3,0.1

Type RM Length L Ch R = 1 ,22034   ,218.8,226.5,236.4
XS GIS Cut Line= 3
2150040.93247463651719.4459190552149883.18353086651890.017015085
 2149782.5139657652081.466167351
#Sta/Elev= 30
       0 1318.36    24.4 1312.96    38.6 1311.88    75.4 1306.35    89.5  1306.5
   105.9 1304.69   122.2 1298.47  135.531291.586   142.5 1289.76   149.5 1289.45
   183.7 1291.49   191.4 1293.43   209.4 1291.45   219.1 1291.96     231 1298.76
   235.9  1299.2   263.6 1293.37   285.6 1292.78   294.7 1294.36   299.2 1298.39
   335.3 1341.42   349.5  1355.2   358.3 1365.61     376 1371.82   393.9 1384.63
   408.7 1387.08   416.7 1392.65   421.2 1394.68   430.2 1401.35   448.6 1409.66
#Mann= 3 ,-1,0
       0      .1       0  135.53    .045       0   183.7      .1       0
Bank Sta=135.53,183.7
XS Rating Curve= 0 ,0
Exp/Cntr=0.3,0.1

Type RM Length L Ch R = 1 ,21808   ,278.2,282.9,269.6
XS GIS Cut Line= 3
2150010.61852779651556.4736381062149724.25246058 651703.94043235
2149629.50229733651873.206285575
#Sta/Elev= 30
       0 1331.27    25.2 1327.18    38.7  1328.6    52.2 1324.12    64.7 1323.44
   119.7 1315.92   141.9  1308.7   155.7  1302.6   169.2 1301.14   180.5 1298.27
   213.2  1293.4     220 1291.11  231.54 1285.16   242.9 1283.26   268.2 1283.03
   281.7 1283.54  289.061285.157   302.3 1291.48   317.7 1291.02   332.7 1295.31
   360.2 1308.96   371.4 1315.87   387.7 1327.57   402.4 1335.65   433.5 1348.77
   447.3 1356.37     461 1362.25   470.2 1365.01   497.7 1378.13   516.1 1381.66
#Mann= 3 ,-1,0
       0      .1       0  231.54    .045       0  289.06      .1       0
Bank Sta=231.54,289.06
XS Rating Curve= 0 ,0
Exp/Cntr=0.3,0.1

Type RM Length L Ch R = 1 ,21525   ,209.2,210.2,205.3
XS GIS Cut Line= 3
2149923.85886162651293.0849778342149569.89786162651494.764977834
2149436.12463042 651721.30456876
#Sta/Elev= 30
       0 1370.33    23.3 1362.57    50.3 1355.25    87.1 1342.11   100.9 1334.53
   110.1 1326.94   120.1 1325.75   143.5    1310   165.4 1299.14   184.6 1294.54
   225.2  1289.6   252.8 1289.63   257.4 1288.57   274.9 1280.52   303.5 1279.04
   319.5 1280.13  364.52 1280.13   369.4 1282.21   381.7 1294.56   392.8 1301.34
   398.7 1303.61   418.6 1306.73   450.1 1308.17   497.3  1312.6   520.9 1316.05
   541.8 1321.64   562.3 1323.23   599.6 1333.21   642.5 1348.49   670.5 1359.86
#Mann= 3 ,-1,0
       0      .1       0   319.5    .045       0  364.52      .1       0
Bank Sta=319.5,364.52
XS Rating Curve= 0 ,0
Exp/Cntr=0.3,0.1

Type RM Length L Ch R = 1 ,21315   ,277.8,254.5,219
XS GIS Cut Line= 4
2149775.02156762651134.9912930252149607.17355303651247.889064746
2149488.28120936651322.8212141182149320.43319477 651651.52357603
#Sta/Elev= 30
       0  1369.8    13.1 1360.56    56.5 1340.08    75.7 1327.23      95 1317.54
   128.8 1312.26   148.1 1296.34   162.1 1280.89   167.3 1277.74   182.3 1275.85
   210.6  1279.1  231.791271.125   253.1 1269.22  294.611271.125   314.6 1271.91
   339.7 1285.44   376.9 1288.13   386.3 1287.32   408.3 1276.56   424.9 1275.41
   435.3  1276.9   462.2 1290.01   478.4 1295.27   536.6 1306.36     570 1310.86
     588 1315.45   600.3 1321.01   682.3 1348.25   695.8 1354.32   711.9 1358.23
#Mann= 3 ,-1,0
       0      .1       0  231.79    .045       0  294.61      .1       0
#XS Ineff= 2 , 0
          207.05 1285.38  382.46         1293.37
Permanent Ineff=
       F       F
Bank Sta=231.79,294.61
XS Rating Curve= 0 ,0
Exp/Cntr(USF)=0,0
Exp/Cntr=0.3,0.1

Type RM Length L Ch R = 1 ,21060   ,259.2,254.8,235.8
XS GIS Cut Line= 3
2149398.61312759651014.1057805172149429.29162011651314.880945582
2149268.60123731651644.195536354
#Sta/Elev= 30
       0 1317.59    15.2 1314.99    31.2 1307.24    55.4 1284.39    67.4 1271.44
    71.4 1268.49   96.531264.415   131.8 1262.77   147.8  1262.8  158.061264.416
     180  1271.7   200.1  1271.9   228.3 1276.41   272.5 1275.15   304.9 1280.16
   319.8 1279.12   344.9 1272.33   376.7  1271.6   406.6  1287.5   420.6 1292.53
   439.5 1296.14   451.5 1300.26   469.6 1299.19   496.3 1303.62   567.5 1330.28
   583.1 1334.73   607.5 1346.47   633.3 1353.02   656.5 1360.65   668.8 1367.17
#Mann= 3 ,-1,0
       0      .1       0   96.53    .045       0  158.06      .1       0
Bank Sta=96.53,158.06
XS Rating Curve= 0 ,0
Exp/Cntr=0.3,0.1

Type RM Length L Ch R = 1 ,20805   ,312.2,359.5,393.5
XS GIS Cut Line= 4
2149341.86209328651024.390517137 2149207.9327159651199.314581722
2149308.04496556651410.8920165562149199.43837175651651.350163218
#Sta/Elev= 30
       0 1303.39    13.2 1301.49    51.4 1291.68   101.5 1283.25   121.9 1281.05
   142.1 1287.38   157.2 1280.57     173 1280.24   198.6 1274.75   230.9 1272.89
   257.9 1260.83   288.7 1257.29     302 1250.36     312 1250.58   332.9 1249.19
   353.8 1250.47   377.3 1252.55   390.1 1255.75   403.8 1262.53   426.6 1279.45
   448.1 1290.12   487.6 1300.62   534.6 1317.79   601.7 1338.39   636.8 1353.08
   658.8 1360.06   676.3  1369.1   702.7 1371.96   711.5 1380.42   718.2 1383.38
#Mann= 3 ,-1,0
       0      .1       0     312    .045       0   353.8      .1       0
Bank Sta=312,353.8
XS Rating Curve= 0 ,0
Exp/Cntr=0.3,0.1

Type RM Length L Ch R = 1 ,20446   ,409.6,421.3,410.1
XS GIS Cut Line= 3
2149278.95902934651054.0224993242149145.87533373651152.850046924
2148680.78368008651300.538972495
#Sta/Elev= 30
       0 1287.36    32.1 1281.42      59 1281.46    73.2 1277.56   127.2 1276.99
   152.9 1274.44   170.6  1274.6   184.3 1269.54   196.9 1267.03   213.7 1259.53
   243.8 1257.39   268.3  1250.9   289.3 1249.53  308.951240.187   318.6 1238.47
   335.4 1238.34  361.611240.186   373.2 1244.32   396.7 1261.34   406.3 1271.32
   415.2 1277.69   436.1 1301.88   457.1 1318.93   478.1 1327.68   514.6 1351.19
   528.5    1358   574.6 1385.71     625 1409.62   637.6 1416.99   653.7 1419.36
#Mann= 3 ,-1,0
       0      .1       0  308.95    .045       0  361.61      .1       0
Bank Sta=308.95,361.61
XS Rating Curve= 0 ,0
Exp/Cntr=0.3,0.1

Type RM Length L Ch R = 1 ,20024   ,401.1,407.1,369.9
XS GIS Cut Line= 3
2149179.77191923 650801.355289062148878.79869727650818.134185904
2148675.33702772650899.215063164
#Sta/Elev= 30
       0 1288.75    47.7 1273.18    59.7 1271.65    67.8  1269.2    75.7  1266.1
    87.7 1259.29    99.8 1253.91   107.8 1248.49   111.8  1247.3   123.8 1247.02
   127.8 1245.65   143.8 1235.96   151.8 1232.41  169.121231.319   183.9 1229.94
   211.9 1229.66  240.941231.322     264 1241.57     280 1251.48     292 1256.89
   312.9 1260.94   321.5 1263.99   338.7  1266.3   347.3 1266.23   360.2 1268.19
   386.1  1270.1     455 1293.49   480.8 1304.51   499.8 1308.98   520.5 1315.32
#Mann= 3 ,-1,0
       0      .1       0  169.12    .045       0  240.94      .1       0
Bank Sta=169.12,240.94
XS Rating Curve= 0 ,0
Exp/Cntr=0.3,0.1

Type RM Length L Ch R = 1 ,19617   ,392.8,410,415.3
XS GIS Cut Line= 3
2149283.75072699650330.9723642812148881.08272699650453.943364281
2148495.13172699650584.654364281
#Sta/Elev= 30
       0 1372.37    12.1 1364.55      33 1359.64    45.6 1349.33    62.3 1340.99
   141.8 1280.97   158.5 1270.12   183.6 1251.35   204.5 1239.54   221.2 1237.59
   271.4 1238.12   321.6 1233.74   363.4 1231.88     376 1229.16   392.3 1229.98
   405.1 1227.33  425.851220.563   468.5 1219.22  507.211220.562   543.3 1238.42
   563.1 1255.62   569.8 1259.59   637.4 1270.12     650 1269.96   679.6 1276.52
   696.5 1278.01   709.2 1282.83   730.3  1286.5   785.2 1292.88   828.5 1302.96
#Mann= 3 ,-1,0
       0      .1       0  425.85    .045       0  507.21      .1       0
Bank Sta=425.85,507.21
XS Rating Curve= 0 ,0
Exp/Cntr=0.3,0.1

Type RM Length L Ch R = 1 ,19207   ,413.6,416.9,404.4
XS GIS Cut Line= 2
2149216.06890952 650090.234786782148434.59012747 650058.25427065
#Sta/Elev= 30
       0 1288.12    23.9  1270.3    47.9 1254.83      76 1238.34      88 1234.01
   235.5 1227.07   280.1 1226.83   289.4  1225.1   308.6 1218.13   332.7 1214.23
   352.2 1215.57   364.2 1210.12  378.161208.697   403.7 1206.33  420.741208.696
   444.3 1211.98   460.3 1216.36   472.3 1223.79   480.3 1231.47   496.3 1241.91
   543.2 1245.06   580.4 1250.24   608.4 1250.32   628.4 1253.48   644.4 1258.43
   660.4 1258.84   712.5 1270.75   732.5 1274.32   744.5 1274.77   782.1  1283.9
#Mann= 3 ,-1,0
       0      .1       0  378.16    .045       0  420.74      .1       0
#XS Ineff= 2 , 0
          348.53 1222.49
Permanent Ineff=
       F       F
Bank Sta=378.16,420.74
XS Rating Curve= 0 ,0
Exp/Cntr=0.3,0.1

Type RM Length L Ch R = 1 ,18790   ,478.5,488.2,462.6
XS GIS Cut Line= 4
2149210.15975846649741.1559394182148956.31186319649670.291002477
2148746.57463808649684.4465468152148450.91524233649779.228970103
#Sta/Elev= 30
       0 1308.17    14.6 1302.94    35.3 1298.85    76.8 1282.59   126.6  1270.6
   147.4 1267.28   176.5 1266.34   188.9 1257.54   193.1 1256.41   263.7 1244.96
   283.7 1244.23   295.8 1238.12   323.8 1208.01  343.071198.797   351.9 1197.15
     384 1196.87  401.581198.796   464.1 1211.27   480.5 1210.18   493.1 1205.57
   514.4 1201.15   530.9 1200.93   564.5 1204.58   585.5  1212.7   598.1 1215.44
   670.3 1213.45   698.9  1215.5   715.7 1218.58   724.4 1222.09   784.2 1257.55
#Mann= 3 ,-1,0
       0      .1       0  343.07    .045       0  401.58      .1       0
#XS Ineff= 2 , 0
                             467         1224.94
Permanent Ineff=
       F       F
Bank Sta=343.07,401.58
XS Rating Curve= 0 ,0
Exp/Cntr=0.3,0.1

Type RM Length L Ch R = 1 ,18302   ,499.7,510.9,508
XS GIS Cut Line= 3
2149232.95818175649505.6010582182148836.00318175649334.646058218
2148546.20593942649271.181630204
#Sta/Elev= 30
       0 1280.87      88 1253.94     101 1252.81   140.2 1240.64   186.6 1231.28
     214 1222.89   231.7 1219.36   275.2 1215.12   336.2  1210.6   349.3  1210.6
   366.7 1208.52   397.2 1200.28   448.4 1199.91     477 1195.91   493.4 1189.31
   509.8 1186.98   522.1 1186.79   538.5  1190.7   554.9 1188.96   571.2 1184.41
   579.4 1183.97   595.8 1185.72   612.2 1183.48  619.511185.942   624.8 1191.48
     645 1222.26   657.2 1238.72   661.3 1243.06   681.9 1253.01   728.9 1288.02
#Mann= 4 ,-1,0
       0     .08       0     200      .1       0   595.8    .045       0
  619.51      .1       0
Bank Sta=595.8,619.51
XS Rating Curve= 0 ,0
Exp/Cntr=0.3,0.1

Type RM Length L Ch R = 1 ,17791   ,490.1,551.2,556
XS GIS Cut Line= 2
2149300.33466719649134.2963335962148824.71318411648841.420607398
#Sta/Elev= 30
       0 1213.32     4.9 1211.19    14.3 1209.89    38.7 1201.54    59.1 1197.42
    75.3 1195.58    89.4 1196.03   139.4 1187.92   166.6 1187.51   178.7 1186.23
   189.9 1188.98   224.8 1189.29   305.5 1186.38   314.9 1184.56   323.6  1179.2
   333.7  1176.4   360.7 1176.15   388.3 1175.04   396.3 1176.28   404.2 1180.48
   416.7 1184.33   427.7 1190.23   432.4 1193.57   441.8 1203.02   451.2 1209.19
   460.5 1217.36   489.4 1231.57   535.7  1262.6   545.1 1266.45   558.6 1269.01
#Mann= 4 ,-1,0
       0     .08       0      70      .1       0   360.7    .045       0
   396.3      .1       0
Bank Sta=360.7,396.3
XS Rating Curve= 0 ,0
Exp/Cntr=0.3,0.1

Type RM Length L Ch R = 1 ,17240   ,493.7,475.5,429.6
BEGIN DESCRIPTION:
XS overtop dirt road
END DESCRIPTION:
XS GIS Cut Line= 6
2149648.84978836648812.1430904792149404.66541388648688.401646083
2149332.92114808648636.1134523612149313.46507599648564.369186556
2149311.03306698648506.000970309 2149132.6971206648450.797086045
#Sta/Elev= 30
       0 1236.32    23.2 1226.59    47.3 1214.62    81.5 1199.69      95 1195.86
   100.9 1192.29   106.9 1190.55   166.7 1185.06   189.1  1184.8   260.8  1179.8
   279.2 1180.57   296.6 1178.34   313.8 1178.69   329.2 1177.13   348.2 1170.32
  354.721169.079   371.3 1167.73   424.5  1167.5   448.9 1167.67  462.55 1169.08
   499.5 1171.79     509    1179   523.8 1185.83   537.1 1190.03   562.3 1193.54
   595.8 1195.76   608.3 1195.09   620.9 1196.34   671.1 1206.92   683.1 1211.19
#Mann= 8 ,-1,0
       0     .08       0      80     .06       0     120     .08       0
     230      .1       0  293.75     .06       0  348.51      .1       0
  354.72    .045       0  462.55      .1       0
Bank Sta=354.72,462.55
XS Rating Curve= 0 ,0
Exp/Cntr=0.3,0.1

Type RM Length L Ch R = 1 ,16765   ,567.5,549,513.7
XS GIS Cut Line= 3
2149960.50224312648462.5230605822149461.68606373648153.520425651
2149200.55787962648191.585694725
#Sta/Elev= 30
       0 1285.49    33.3 1271.17    66.3 1251.97    75.7 1245.28    86.1  1233.9
   103.9 1231.98   108.6 1230.35   155.7 1198.18   169.7 1186.46   179.2  1185.2
   198.8 1173.58   207.4  1171.1   226.2 1169.94   320.8 1169.74   329.2 1168.18
  347.611161.256   372.1  1159.3  402.461161.255   434.1 1165.28   456.8  1164.3
   470.9 1162.24     501 1167.08   541.6 1167.91   560.3 1171.12     616 1171.54
   677.2 1174.51   693.6 1176.98   782.3 1183.04   818.7  1187.2   850.7 1193.12
#Mann= 6 ,-1,0
       0     .06       0     150      .1       0  347.61    .045       0
  402.46      .1       0  606.77     .06       0  706.77      .1       0
Bank Sta=347.61,402.46
XS Rating Curve= 0 ,0
Exp/Cntr=0.3,0.1

Type RM Length L Ch R = 1 ,16216   ,524.7,507.5,468.9
XS GIS Cut Line= 5
2149891.88928702647606.3873556272149777.44948709647760.595455706
2149608.25867962647806.7913855242149409.35331086647988.689240123
2149228.11373942648015.947413845
#Sta/Elev= 30
       0 1240.14    27.5 1231.03    41.8  1229.5    56.1 1225.24    93.3 1217.49
     123 1208.33   167.6 1188.62   201.6 1177.62   206.6    1175   226.5 1158.95
  242.511153.568     268 1150.31   292.9  1149.5   309.5 1149.76  321.751153.568
   334.3 1159.32   350.9 1162.62   448.8 1161.73   505.1 1165.17   524.9 1164.87
   558.9 1161.32   596.2 1160.61   627.7 1165.99   654.3    1168   666.5 1170.44
     719 1176.14   755.5 1175.72   771.6 1178.29     804 1178.27   820.2 1181.52
#Mann= 5 ,-1,0
       0      .1       0  242.51    .045       0  321.75      .1       0
  587.42     .06       0  706.95      .1       0
#XS Ineff= 2 , 0
                          523.93         1167.49
Permanent Ineff=
       F       F
Bank Sta=242.51,321.75
XS Rating Curve= 0 ,0
Exp/Cntr=0.3,0.1

Type RM Length L Ch R = 1 ,15708   ,482.4,482.3,435.3
XS GIS Cut Line= 3
2149510.01558805647228.5951930752149275.37639277647571.461311722
 2149045.0349742 647799.41359764
#Sta/Elev= 30
       0 1246.16      54 1226.95      88 1213.91    95.3 1210.26   108.2 1208.15
   112.2  1206.5   121.9 1200.92   165.8 1163.89   175.2 1159.37     183 1154.16
   184.9 1153.42   204.3 1154.17  217.241151.378   223.3 1149.91   240.6 1149.34
  281.411151.377     340 1156.13   369.1 1155.73   398.2 1157.21   549.1  1155.4
   560.1 1157.87   565.8 1160.27   582.8 1171.45   605.6 1181.29   616.9 1187.56
   628.3 1189.16   645.2 1194.31   693.3 1202.07   707.4 1205.63   739.5 1211.05
#Mann= 5 ,-1,0
       0      .1       0  217.24    .045       0  281.41      .1       0
  455.47     .06       0  595.47      .1       0
#XS Ineff= 2 , 0
                          414.67          1173.2
Permanent Ineff=
       F       F
Bank Sta=217.24,281.41
XS Rating Curve= 0 ,0
Exp/Cntr=0.3,0.1

Type RM Length L Ch R = 1 ,15226   ,494.8,510.3,509.2
XS GIS Cut Line= 4
2149033.36161164647023.6334001552148948.01951141647269.606941779
2148947.67744234647495.1071474942148856.54324391647761.816044217
#Sta/Elev= 30
       0 1227.48   141.4 1179.43   162.5 1168.52   187.9 1158.66   221.8 1151.35
   247.2 1150.44   271.9    1151   275.9 1150.41   294.71143.005   299.9 1141.47
   323.9 1141.08   339.9 1142.95   355.9 1143.78   379.9 1141.43   391.9 1143.41
   411.9 1148.94   443.9 1149.61   475.9 1153.23     488 1153.14   509.2 1151.15
   526.1  1151.2   543.8 1152.93   591.1 1164.56   606.4 1170.73   628.9 1182.13
   644.4 1184.64   657.1 1192.05   669.9 1196.27   717.1 1215.22   767.7  1229.8
#Mann= 5 ,-1,0
       0      .1       0   294.7    .045       0   339.9      .1       0
  495.86     .06       0  595.86      .1       0
Bank Sta=294.7,339.9
XS Rating Curve= 0 ,0
Exp/Cntr=0.3,0.1

Type RM Length L Ch R = 1 ,14716   ,406.7,422.8,419.7
XS GIS Cut Line= 3
     2148723.813      646917.4092148536.37214886647247.387913772
2148357.43906263647508.944827543
#Sta/Elev= 30
       0 1223.62    77.9 1203.18   114.7 1190.49   125.7 1188.63     145 1182.44
   166.8 1172.43   202.1 1151.17   217.9 1145.09   240.1 1142.07   295.9 1145.95
   348.7 1146.59   406.8 1144.96   475.9 1137.12   493.2 1134.94  507.121137.177
   516.2 1137.52   527.1 1135.43   533.5 1136.02   539.2 1138.51   546.4 1143.77
   575.5 1174.98   590.1 1187.65   604.6 1197.95   625.5 1208.19   639.9 1209.29
   643.4 1211.21   648.2 1216.58   653.1 1220.23   665.8 1223.09   696.4 1239.21
#Mann= 5 ,-1,0
       0      .1       0   475.9    .045       0  507.12      .1       0
   519.5     .06       0   569.5      .1       0
#XS Ineff= 2 , 0
          307.48 1165.44
Permanent Ineff=
       F       F
Bank Sta=475.9,507.12
XS Rating Curve= 0 ,0
Exp/Cntr=0.3,0.1

Type RM Length L Ch R = 1 ,14293   ,417.7,413.8,392
XS GIS Cut Line= 4
 2148490.8259742646774.4124789942148352.48177451646949.941076634
2148155.13805982647060.6120840892148024.14043037647239.334790716
#Sta/Elev= 30
       0 1242.45    13.7 1235.74    30.1 1229.97    64.6  1212.9    79.9 1206.89
   100.3 1197.11   115.6 1187.51   130.8 1181.49   180.4 1151.89   197.5 1144.59
   223.2 1139.02   260.5 1138.18   274.3  1135.1   283.5 1131.66  295.14  1130.7
   301.8 1128.91   324.7 1128.58   347.7 1130.68     366 1130.62   388.9  1134.9
   411.2  1141.2   425.6 1143.08     510 1146.94   552.4 1163.55   564.5 1165.47
   569.5 1167.64   583.3 1176.35   595.4 1179.47     634 1193.58   671.3 1209.22
#Mann= 4 ,-1,0
       0      .1       0  295.14    .045       0   347.7     .06       0
  443.49      .1       0
Bank Sta=295.14,347.7
XS Rating Curve= 0 ,0
Exp/Cntr=0.3,0.1

Type RM Length L Ch R = 1 ,13879   ,441.6,428,405.6
XS GIS Cut Line= 3
2148187.38379292646459.3349675822147950.05879292646790.521967583
2147715.79207663647040.952462785
#Sta/Elev= 30
       0 1291.65      22 1280.61    56.4 1261.24    71.2 1254.02    83.9 1246.36
    94.8 1237.98   105.6 1234.01   159.7 1198.65   194.2 1181.77   211.5 1168.95
   218.4 1162.79     233 1144.81   238.7 1135.61   243.4 1129.71   248.3 1127.31
  257.251125.645   287.4 1123.19   297.5 1123.39  311.991125.646   346.7 1128.66
   361.5 1133.82   376.3 1136.85   403.8 1136.67   416.3 1140.73   461.6 1145.08
   527.3 1149.59   563.5 1154.69   656.9 1170.29   723.3 1185.62   750.4 1194.39
#Mann= 5 ,-1,0
       0      .1       0  257.25    .045       0  311.99      .1       0
     320     .06       0  437.44      .1       0
Bank Sta=257.25,311.99
XS Rating Curve= 0 ,0
Exp/Cntr=0.3,0.1

Type RM Length L Ch R = 1 ,13451   ,578.6,612.7,612.2
XS GIS Cut Line= 3
2147633.95590936646358.4077560932147617.43449162646700.019406836
     2147620.665      646999.623
#Sta/Elev= 30
       0 1214.45    30.8 1203.04    50.8 1197.76    66.8 1191.63    78.9 1188.87
    90.9 1182.34   126.6  1154.6   153.3 1127.44     159 1122.45  163.981119.338
     167 1118.16     207 1117.09     231 1117.98  237.981119.337   247.1 1122.81
   255.1 1123.46   267.1 1127.73   279.1 1128.98   291.1 1128.67   323.1 1131.85
   395.2 1131.89   411.2    1139   425.3 1146.95   435.2 1150.54   447.2 1152.42
   483.2 1155.22   543.2 1167.42   571.2 1177.26   579.2 1178.89   641.6 1196.83
#Mann= 5 ,-1,0
       0      .1       0     160     .06       0  163.98    .045       0
  237.98     .06       0     260      .1       0
Bank Sta=163.98,237.98
XS Rating Curve= 0 ,0
Exp/Cntr=0.3,0.1

Type RM Length L Ch R = 1 ,12838   ,467,471.7,472.3
XS GIS Cut Line= 3
  2147308.495986646209.786923366  2147053.976986646529.176923366
  2146817.540986646873.879923366
#Sta/Elev= 30
       0 1215.46    13.4 1205.38   101.5    1158   111.7 1154.31     122 1148.14
   133.6 1146.67   156.4 1137.22   188.5 1130.53   210.4 1114.01   239.6 1112.55
   263.7 1116.34   290.8  1114.4  305.211110.438   321.4 1108.09  349.841110.439
   372.8  1111.5   404.9 1117.67   418.1 1118.51   534.5 1115.38   547.8 1115.91
   558.8 1118.98   587.9 1138.84   608.2 1155.88   612.1 1160.11   621.8 1176.43
   631.2 1184.58     660 1198.46   734.8 1246.11   766.5 1259.52   826.4 1290.39
#Mann= 3 ,-1,0
       0      .1       0  305.21    .045       0  349.84      .1       0
#XS Ineff= 2 , 0
                          455.79         1126.63
Permanent Ineff=
       F       F
Bank Sta=305.21,349.84
XS Rating Curve= 0 ,0
Exp/Cntr=0.3,0.1

Type RM Length L Ch R = 1 ,12367   ,307,342.5,345.4
XS GIS Cut Line= 4
2146848.43500661646098.2690722252146707.67063452646259.153448073
2146620.83272511646445.1542372922146511.97856004646633.716943984
#Sta/Elev= 30
       0 1154.91     7.9 1152.77    24.9 1142.05    56.1 1126.18    62.3 1123.98
    73.1 1121.35   180.8  1117.2   206.9 1116.72     236 1112.45   246.9 1111.64
   251.3 1110.65   260.2 1106.43   270.51105.106   361.7 1102.62   370.5 1103.02
  384.281105.104   392.5 1107.44   410.2 1114.86   419.1 1115.24   423.7 1116.35
   428.3 1119.46   437.5 1127.12   446.8 1131.83     481 1156.46   530.8 1186.09
   548.4 1200.34   574.7 1218.07   592.1 1228.15   618.7 1242.33   636.8 1249.44
#Mann= 4 ,-1,0
       0      .1       0   270.5    .045       0  384.28     .06       0
  393.77      .1       0
Bank Sta=270.5,384.28
XS Rating Curve= 0 ,0
Exp/Cntr=0.3,0.1

Type RM Length L Ch R = 1 ,12024   ,409.5,416.5,405.3
XS GIS Cut Line= 4
     2146754.993      645898.6642146566.63550085646085.248741897
2146375.02423985646192.0107842232146183.85994199646430.235387759
#Sta/Elev= 30
       0 1236.61     9.3 1233.28    20.7 1226.17    32.1 1224.36    97.1 1185.69
   108.4 1183.41   122.6 1173.95   159.3 1156.45   210.2 1129.68   238.5  1117.2
     265 1109.82   277.1 1108.83   290.8 1105.39   336.6 1104.92   352.2 1101.92
   368.7 1101.03   419.1 1101.16   437.1 1099.94  453.931101.304     458 1103.49
   469.8 1113.37   483.2 1114.98   537.3 1128.82   609.1 1158.41   666.6 1187.57
   711.6 1215.76   731.9 1226.78   738.3 1232.33   762.9 1244.18   789.9 1254.04
#Mann= 5 ,-1,0
       0      .1       0  355.13     .06       0   419.1    .045       0
  453.93     .06       0  465.13      .1       0
Bank Sta=419.1,453.93
XS Rating Curve= 0 ,0
Exp/Cntr(USF)=0,0
Exp/Cntr=0.3,0.1

Type RM Length L Ch R = 1 ,11608   ,496.3,512.7,499
XS GIS Cut Line= 2
2146415.90888356645673.9527140822145883.26859025646089.162918956
#Sta/Elev= 30
       0 1230.24    19.9 1215.55    47.7  1196.7    81.9 1176.37      96 1164.13
   110.4  1161.2   115.9 1157.83   128.9 1146.92   140.9 1140.26   148.4 1137.86
   153.2 1134.14     167 1119.17     176 1117.25   187.3 1112.18   201.6 1108.43
   215.9  1101.6  242.241098.687   273.5 1093.99   278.6 1094.31  293.691098.686
     309 1100.38   319.2 1100.45   352.7 1104.97   441.2 1108.42   471.3 1111.67
   486.6  1114.3   511.9 1122.22   577.8 1146.49   649.4 1177.88   675.4 1190.38
#Mann= 6 ,-1,0
       0      .1       0     160     .06       0  242.24    .045       0
  293.69      .1       0     410     .08       0     570      .1       0
Bank Sta=242.24,293.69
XS Rating Curve= 0 ,0
Exp/Cntr=0.3,0.1

Type RM Length L Ch R = 1 ,11095   ,461.4,465.2,454.7
XS GIS Cut Line= 2
2146062.24828812645356.8935630182145576.62217389645723.577949169
#Sta/Elev= 30
       0 1164.38    12.6 1159.07    22.6 1156.09    37.7 1146.36    47.7 1145.17
    52.7 1143.31    67.8  1135.1    84.5 1123.74    97.8 1119.22   121.6 1103.43
   130.2  1099.9   133.1 1099.07   141.6  1099.2     153 1094.48     158 1093.72
   167.3 1096.06   181.6 1095.08   195.9 1097.14   206.3 1096.09   226.2 1092.49
   240.1 1096.11   246.1  1098.9   255.9 1099.08   264.4 1101.63   441.5  1098.5
     470 1099.77   478.8 1102.94   493.8  1111.2   551.4 1147.67   608.5 1172.65
#Mann= 5 ,-1,0
       0      .1       0      80     .06       0     200      .1       0
   206.3    .045       0   240.1      .1       0
Bank Sta=206.3,240.1
XS Rating Curve= 0 ,0
Exp/Cntr=0.3,0.1

Type RM Length L Ch R = 1 ,10630   ,430.6,435.1,415.2
XS GIS Cut Line= 3
2145724.89653942644982.6404443722145562.17783714645261.083760503
2145385.16379292645586.799776712
#Sta/Elev= 30
       0 1137.49    26.1 1130.07    35.4 1128.69    46.2  1123.7    67.8 1118.34
      91 1116.13   104.9 1116.08   109.5 1114.79     128 1104.59   139.8 1099.89
   160.5 1099.64   192.9 1094.35   212.9 1094.12   223.4  1094.8   253.1 1093.11
   277.3 1091.75     286 1093.13   304.1 1094.79   318.2 1098.22     377 1098.03
   427.3 1096.84   460.7 1091.78   498.1 1090.53   509.3 1091.96   515.8 1094.09
   582.1  1130.8   594.8 1134.43   609.4 1141.22   668.6 1161.91   693.2 1171.53
#Mann= 5 ,-1,0
       0      .1       0     180     .06       0   253.1    .045       0
     286     .06       0     300      .1       0
Bank Sta=253.1,286
XS Rating Curve= 0 ,0
Exp/Cntr=0.3,0.1

Type RM Length L Ch R = 1 ,10194   ,505,511,493.2
XS GIS Cut Line= 3
2145249.46719528644826.8473397292145194.89906043645164.719386151
2145075.67039056645586.911818723
#Sta/Elev= 30
       0 1198.74    38.8 1180.73    79.3 1153.72    91.5 1150.64   115.8 1134.24
   140.1 1113.51   172.5 1091.34   198.5 1089.65   225.2 1090.42  235.61 1087.81
   265.7 1085.85   310.3 1086.09  320.621087.874   326.5 1089.36   334.6 1093.75
   338.7 1094.41     351 1092.35   405.1 1092.68   475.7 1090.14   492.4 1086.92
   506.9 1088.73   526.3 1088.82   542.2 1097.11   567.2 1116.53   583.8 1127.89
   604.6 1138.94   661.4 1161.81   725.1 1191.77   758.4 1203.77     781 1210.19
#Mann= 5 ,-1,0
       0      .1       0     230     .05       0  235.61    .045       0
  320.62     .06       0  422.25      .1       0
Bank Sta=235.61,320.62
XS Rating Curve= 0 ,0
Exp/Cntr=0.3,0.1

Type RM Length L Ch R = 1 ,9683    ,526.9,538.4,510.8
XS GIS Cut Line= 2
2144723.77766148644849.5038435922144680.93955684645527.797608505
#Sta/Elev= 30
       0 1155.35    35.7 1143.51    51.8 1140.37    75.8  1131.5   111.9 1120.16
   127.9 1116.69   158.4 1107.23     164 1104.19     172 1097.91     184 1085.75
  187.661082.995   192.1 1081.79   244.2 1080.76     267 1082.98   280.2 1083.41
   292.3 1082.22   312.4 1083.92   320.9 1085.72   380.1 1087.38   396.5 1086.76
   424.5 1083.42   444.6 1083.03   476.6 1087.45   480.6 1088.83   488.6 1095.27
   516.7 1113.88   548.8 1131.78   576.8 1149.23   600.9  1162.4   679.6 1212.84
#Mann= 5 ,-1,0
       0      .1       0  187.66    .045       0     267      .1       0
     390     .06       0     490      .1       0
Bank Sta=187.66,267
XS Rating Curve= 0 ,0
Exp/Cntr=0.3,0.1

Type RM Length L Ch R = 1 ,9145    ,564.9,584.6,594.8
XS GIS Cut Line= 3
2144363.13047109644791.5635227012144270.03198722645074.412888558
2144155.94583459645493.939645441
#Sta/Elev= 30
       0 1130.12    35.4 1116.55    81.7 1101.67     107 1094.64   146.2 1086.03
   165.9 1080.18   178.6 1080.09   195.4 1082.47   258.6 1084.75   333.8 1084.65
   371.1 1082.99   376.5 1081.57  385.221076.638     396 1073.88  436.39 1076.64
   441.7 1079.64     454 1095.58   458.2 1099.92     471 1117.11     483 1127.65
   503.8 1142.05   516.2 1143.36   520.3 1144.96   528.6 1151.51   549.4 1158.52
   570.1 1167.32   640.5 1201.62   648.8 1204.52   665.4  1212.5   732.5 1238.49
#Mann= 7 ,-1,0
       0      .1       0  367.78     .06       0  385.22    .045       0
  436.39     .06       0  457.78      .1       0  467.78     .06       0
  567.78      .1       0
Bank Sta=385.22,436.39
XS Rating Curve= 0 ,0
Exp/Cntr=0.3,0.1

Type RM Length L Ch R = 1 ,8561    ,490.4,488.2,467.8
XS GIS Cut Line= 3
     2144035.029      644601.119     2143756.056      644901.115
     2143478.092      645208.575
#Sta/Elev= 30
       0 1125.19    49.2 1109.12   109.9 1086.36   133.4 1080.48   152.1 1078.78
   227.4 1077.39   355.1 1079.28   362.5 1077.89  370.641072.774   384.2  1070.8
   409.6 1070.53   454.9 1071.16   464.41072.778   469.1 1074.61   474.5 1078.87
     493  1096.7   534.2 1120.54   540.7 1123.34   549.9 1123.84   556.9 1126.23
   614.7 1153.98     639 1154.38   653.2 1158.77   671.9  1161.7   709.8 1172.15
     724 1174.81   743.5 1185.72   761.4 1188.72   780.6 1198.05   824.1 1208.33
#Mann= 5 ,-1,0
       0      .1       0  370.64    .045       0   464.4      .1       0
  469.66     .06       0  599.66      .1       0
#XS Ineff= 2 , 0
          196.76  1086.8
Permanent Ineff=
       F       F
Bank Sta=370.64,464.4
XS Rating Curve= 0 ,0
Exp/Cntr=0.3,0.1

Type RM Length L Ch R = 1 ,8072    ,430.9,441.9,423.1
XS GIS Cut Line= 3
2143549.90197404644248.7523957542143518.88392258644321.259946918
2143285.56278757644963.252302911
#Sta/Elev= 30
       0 1099.65    52.7 1079.15    65.7 1077.53    87.3 1077.08   108.6 1072.75
   142.6 1071.92   265.1  1073.3  294.061070.085   309.3  1067.1   329.9 1067.38
  358.021070.086   389.5 1072.39   410.7 1075.28   435.2 1073.94   458.6 1073.82
   483.6 1075.57   495.9 1077.88   539.8 1095.47   592.8    1120   610.8 1127.73
   623.5 1131.91   644.8 1141.85   649.1 1142.84   658.4 1142.94   670.4 1147.99
   683.1 1148.82   691.6 1153.47     699 1155.35   745.8 1163.36   761.9 1167.53
#Mann= 5 ,-1,0
       0      .1       0  294.06    .045       0  358.02      .1       0
  538.86     .06       0  638.86      .1       0
Bank Sta=294.06,358.02
XS Rating Curve= 0 ,0
Exp/Cntr=0.3,0.1

Type RM Length L Ch R = 1 ,7630    ,698.7,695.2,657.7
XS GIS Cut Line= 3
2143153.21757435644129.382450033 2143057.0126963644662.983538936
2143114.77920928644931.787298971
#Sta/Elev= 30
       0 1106.34    56.7  1095.7    68.9 1094.99    97.3 1088.27   101.4 1086.38
   105.5 1082.86  117.831067.378   121.7  1064.6   129.9 1063.45  172.411067.381
   219.3 1071.69   243.7  1070.7   308.7 1072.09   410.3 1071.79   487.5 1069.72
   503.8    1071   511.9 1073.03     529 1079.99   556.7 1089.11   564.9 1090.76
   598.3 1101.44   618.1    1109   634.5 1114.02     659 1123.94   675.4 1124.63
   687.6 1133.11   699.9 1137.56     749 1151.01   769.5 1154.56   817.1 1167.01
#Mann= 7 ,-1,0
       0      .1       0  117.83    .045       0  172.41      .1       0
     230     .05       0     430      .1       0     530     .06       0
   632.2      .1       0
Bank Sta=117.83,172.41
XS Rating Curve= 0 ,0
Exp/Cntr=0.3,0.1

Type RM Length L Ch R = 1 ,6935    ,507.6,504.7,488.2
XS GIS Cut Line= 3
2142424.35205822644203.628663252 2142701.2615114 644873.96553736
2142797.04281589645007.757268286
#Sta/Elev= 30
       0 1114.44    53.6 1101.47    62.3 1098.07    86.8 1078.31  101.171063.088
   105.5 1061.37   148.8 1060.77  172.051063.083     194 1066.96   203.2 1067.56
   249.1 1066.24   287.3 1067.25   425.8  1066.7   482.1 1067.75   551.3 1065.82
   596.7  1067.7   668.2 1067.96   690.2  1069.2   698.5 1071.64   715.8 1081.79
   729.2 1083.32   734.2 1085.41     744 1094.71   753.8 1100.91     803 1125.15
   827.1 1135.93     854 1144.81   871.9 1153.03   881.5 1155.62   889.8 1159.76
#Mann= 6 ,-1,0
       0      .1       0  101.17    .045       0  172.05     .05       0
     610      .1       0     700     .06       0  815.28      .1       0
Bank Sta=101.17,172.05
XS Rating Curve= 0 ,0
Exp/Cntr=0.3,0.1

Type RM Length L Ch R = 1 ,6431    ,562.9,599.3,632.8
XS GIS Cut Line= 4
2142017.44426986644334.1716955132142000.88046077644519.465580273
2142347.70742014644968.0763272922142402.34754445645131.248450821
#Sta/Elev= 30
       0 1088.75    23.1 1086.51    55.2 1082.01    63.3 1080.01    87.4 1078.25
   139.6 1072.14   206.7 1066.33   223.8 1067.42   230.7 1065.69  243.221058.684
   250.3    1057   289.3 1056.81   309.4 1057.45  313.781058.684   329.3  1063.2
   340.7  1063.8   420.8 1061.69   476.4 1061.77   511.8 1063.12   534.6 1065.12
   587.6 1064.81   642.7  1066.8   728.5 1067.68   762.7 1069.58   771.1 1073.51
   813.3 1101.85   839.6  1126.7     847  1132.5   905.7 1161.75   925.2 1169.49
#Mann= 5 ,-1,0
       0      .1       0  243.22    .045       0  313.78      .1       0
  726.03     .06       0  793.08      .1       0
Bank Sta=243.22,313.78
XS Rating Curve= 0 ,0
Exp/Cntr=0.3,0.1

Type RM Length L Ch R = 1 ,5831    ,617.3,614.2,619.2
XS GIS Cut Line= 3
 2141753.2147561      644327.8812141607.07512116 644780.77266798
 2141484.3406963645088.052032261
#Sta/Elev= 30
       0 1092.41      77 1073.11    87.7 1069.39   106.4 1060.86   114.8 1059.05
   131.7 1059.75   169.5  1059.1   186.2 1060.77   207.3    1060   291.4 1061.46
   413.3 1061.33   476.3 1062.23   481.5 1061.68   497.9 1056.15   502.2 1055.93
   512.3 1057.83  525.09 1055.94   546.1 1052.33   571.1 1052.53   579.7 1054.22
   589.2 1054.59  594.331055.947   601.2 1059.37   618.5 1076.49   627.1 1081.93
   631.4 1083.74   690.8 1100.98   709.3 1105.63   721.6 1107.52   806.8 1128.01
#Mann= 3 ,-1,0
       0      .1       0  525.09    .045       0  594.33     .05       0
Bank Sta=525.09,594.33
XS Rating Curve= 0 ,0
Exp/Cntr=0.3,0.1

Type RM Length L Ch R = 1 ,5217    ,418.3,439.4,426.8
XS GIS Cut Line= 2
2141242.51944798644109.0004485612140992.78522784644897.208535034
#Sta/Elev= 30
       0 1105.84     8.6 1098.95    25.4 1082.64      38 1072.64    54.7 1057.12
    58.9 1054.59    71.5 1051.88    88.3 1052.21   100.9 1051.34   113.7 1052.98
   159.6  1053.6   184.8 1052.59   285.6  1055.5   323.3 1053.66   369.4 1052.58
  382.331053.637   391.8 1055.11   419.8 1054.81   449.2 1056.93   511.8  1056.5
   549.9 1055.65   558.3 1057.77   570.8 1063.39   585.1 1066.42   650.6 1074.25
   775.9 1090.84     789 1093.46   805.8 1097.99   818.4 1100.12   826.8 1102.57
#Mann= 3 ,-1,0
       0      .1       0   323.3    .045       0  382.33      .1       0
Bank Sta=323.3,382.33
XS Rating Curve= 0 ,0
Exp/Cntr=0.3,0.1

Type RM Length L Ch R = 1 ,4778    ,605.1,605.9,593.4
XS GIS Cut Line= 3
2140934.59300487644023.2331371212140706.51430792644530.318154854
2140679.48319406644784.311471128
#Sta/Elev= 30
       0 1098.92    10.9 1085.99    28.4 1070.34    50.4 1059.21   59.611049.708
    63.5 1048.24    81.1 1047.95     103 1048.31 116.6191049.636   130.4 1050.03
   152.2 1047.99   168.8 1049.01   196.9  1052.8   326.7 1054.07   345.2 1053.07
   366.2 1050.51   381.5 1052.15   453.9 1050.44     467 1051.42   497.8 1047.55
   515.3 1047.23   519.7 1047.63   522.7 1049.16   532.8 1057.98   537.2 1060.23
   554.8 1063.71   623.3 1066.81   671.5 1071.57   745.7 1082.16   811.4 1092.85
#Mann= 5 ,-1,0
       0      .1       0   59.61    .045       0 116.619      .1       0
     370     .05       0  676.02      .1       0
Bank Sta=59.61,116.619
XS Rating Curve= 0 ,0
Exp/Cntr=0.3,0.1

Type RM Length L Ch R = 1 ,4172    ,500.8,508.8,514.3
XS GIS Cut Line= 3
2140352.86237902 643881.272912082140248.24879732644328.871865043
2140268.97818992644756.615713194
#Sta/Elev= 30
       0 1128.23    12.2 1124.39    45.1 1106.08    73.8 1088.31   102.6 1069.66
   123.1 1051.85  130.951046.321     137 1044.46   164.2 1044.31   184.8 1044.54
   191.9 1046.34   209.4 1047.41   221.7 1049.61   260.2 1049.74     308 1047.76
   320.3 1044.58   328.5 1043.97   336.8 1044.38   349.1 1048.05     386 1048.27
     472 1058.66     512  1060.7   532.1 1065.08   548.1 1061.53   652.2 1061.44
   676.2 1065.13   736.3 1067.26   784.1 1073.05   848.4 1078.67   887.9 1085.96
#Mann= 7 ,-1,0
       0      .1       0  130.95    .045       0   191.9      .1       0
     280     .05       0  489.66     .03       0  589.66     .05       0
  779.66      .1       0
Bank Sta=130.95,191.9
XS Rating Curve= 0 ,0
Exp/Cntr=0.3,0.1

Type RM Length L Ch R = 1 ,3663    ,595.8,574.7,557.2
XS GIS Cut Line= 2
2139915.56053986643724.6534204932139514.87570112644527.406382475
#Sta/Elev= 30
       0  1088.8    32.7 1077.18    52.4 1074.83    76.6 1063.89    92.4 1060.93
  115.271043.909   121.3 1041.56   143.6 1041.17     158 1041.54  166.591043.904
   174.9 1044.74   186.7 1042.83   196.8 1043.51   206.2 1041.79   219.6  1044.7
   237.5 1044.56   255.4 1042.58   268.3 1044.31   282.2 1044.28   295.6 1049.33
   331.4  1047.8     470 1047.05   599.3 1048.28   613.1 1049.77   635.4 1056.43
   644.4 1057.77   697.7 1056.15   742.5 1056.78   809.8 1059.99   897.2 1067.19
#Mann= 6 ,-1,0
       0      .1       0  115.27    .045       0  166.59      .1       0
     370     .05       0     590     .06       0     810     .05       0
Bank Sta=115.27,166.59
XS Rating Curve= 0 ,0
Exp/Cntr=0.3,0.1

Type RM Length L Ch R = 1 ,3088    ,562,564.3,567.6
XS GIS Cut Line= 2
 2139246.9190142 643646.673007442139448.31718143644555.391346636
#Sta/Elev= 30
       0 1123.23     5.8 1119.61    16.6 1116.47    27.1  1110.2    39.4 1106.25
   100.4 1096.88   113.2 1093.93   117.3 1091.45   141.9 1070.61   154.2 1061.39
   162.4  1053.8   170.5 1044.69   174.2 1041.82   178.7 1040.17   186.9 1039.36
   211.5 1039.28     232 1039.43  246.671041.844   268.9 1040.82   284.9 1041.36
   305.7 1044.18     318 1044.94   365.4 1045.07   383.6 1044.01     441 1044.77
   575.4 1050.34   645.8 1053.91   690.9 1057.15   724.2 1057.93   930.8 1069.22
#Mann= 9 ,-1,0
       0      .1       0   174.2    .045       0  246.67      .1       0
     290     .05       0     320     .06       0     420     .05       0
     520     .06       0     730     .05       0     930     .06       0
Bank Sta=174.2,246.67
XS Rating Curve= 0 ,0
Exp/Cntr=0.3,0.1

Type RM Length L Ch R = 1 ,2524    ,827,831.2,801
XS GIS Cut Line= 2
2138699.89038851643693.8193029932138836.53707868644619.481210752
#Sta/Elev= 30
       0 1115.29    11.5 1105.82    27.9 1102.36    43.8 1089.28      56 1082.24
    68.1 1072.39    98.3 1052.32   108.9 1047.85   140.9 1040.32     157 1041.19
   169.2 1039.93   221.7 1042.13   244.61040.231   254.1 1038.54     271 1038.28
   310.7 1038.53  322.481040.219     335 1041.55   359.2 1040.28   460.3 1041.64
   517.6 1040.57   545.2 1042.79   625.1 1043.41   747.4 1042.31   763.5 1044.46
   783.8 1051.12     804  1055.6   892.9 1070.22   921.2 1078.43   935.7 1084.24
#Mann= 6 ,-1,0
       0      .1       0   244.6    .045       0  322.48      .1       0
     770     .06       0     800      .1       0     870     .06       0
Bank Sta=244.6,322.48
XS Rating Curve= 0 ,0
Exp/Cntr=0.3,0.1

Type RM Length L Ch R = 1 ,1693    ,390,399.5,383.6
XS GIS Cut Line= 3
2137931.96535422643834.0204247712138156.37657968644306.193116436
2138137.13704144644599.650693149
#Sta/Elev= 30
       0 1088.16     7.9 1086.29    37.8 1083.83    47.8 1079.97    61.1 1077.86
    78.8 1071.65    87.6  1065.9   100.9 1052.73   114.2 1042.91  131.021036.243
   140.6 1033.93   158.5 1033.12   179.6 1033.32  194.991036.242   207.2 1038.72
   252.1 1040.62   348.9 1040.04   415.4 1037.72   446.4 1038.77   459.7 1042.52
   476.8 1045.05   601.9 1055.98   690.1  1067.5   702.2 1069.97   726.2 1069.82
   730.2 1070.95   738.2 1075.91   774.6 1084.68   802.4  1093.3   816.9  1099.2
#Mann= 5 ,-1,0
       0      .1       0  131.02    .045       0  194.99      .1       0
  572.79     .06       0  772.79      .1       0
Bank Sta=131.02,194.99
XS Rating Curve= 0 ,0
Exp/Cntr=0.3,0.1

Type RM Length L Ch R = 1 ,1293    ,430.6,447.8,450.1
XS GIS Cut Line= 2
2137561.70531556643930.9156777842137955.51640977644655.130891724
#Sta/Elev= 30
       0 1099.03    12.3  1092.9    27.1 1091.28    70.9    1068    97.9 1057.43
   133.3 1050.11   152.8 1037.57   166.5 1036.51   202.9 1036.77214.27391034.646
   221.7 1032.83   233.5  1032.3   274.8 1032.69   294.31034.626   312.2 1037.08
   330.4 1035.71   348.6 1037.16   407.6    1037   471.5 1038.43     549 1043.24
   581.6 1047.11   635.5 1047.69   649.9 1050.75   684.8 1053.34   699.2 1056.05
   717.4 1056.15     768 1070.53   799.4 1081.59   811.6 1088.23   824.4 1089.74
#Mann= 5 ,-1,0
       0      .1       0214.2739    .045       0   294.3      .1       0
     710     .06       0     780      .1       0
Bank Sta=214.2739,294.3
XS Rating Curve= 0 ,0
Exp/Cntr=0.3,0.1

Type RM Length L Ch R = 1 ,846     ,394.2,426.5,430
XS GIS Cut Line= 3
2137194.21909351644050.0387994452137398.71696919644646.053975583
2137603.21484488644911.726429462
#Sta/Elev= 30
       0 1110.36    20.2 1102.82    49.8 1085.29    58.3 1082.02    75.2 1077.39
      89 1076.35   104.8 1069.37   151.3 1059.82   180.9 1049.68   214.8 1043.43
   227.6 1039.64   244.4 1032.08   262.2 1032.81   307.8 1030.53     367 1030.82
  380.541032.752   392.4 1036.76   434.7 1034.78   586.9 1035.22   620.7 1040.95
   701.8 1043.09   747.5 1046.27   770.3 1052.41   787.4 1053.73   795.6 1058.47
   870.1 1087.86   915.8 1104.19   931.9 1111.47     942    1113   965.4 1124.33
#Mann= 5 ,-1,0
       0      .1       0   262.2    .045       0  380.54      .1       0
  760.12     .06       0  860.12      .1       0
Bank Sta=262.2,380.54
XS Rating Curve= 0 ,0
Exp/Cntr(USF)=0,0
Exp/Cntr=0.3,0.1

Type RM Length L Ch R = 1 ,419     ,408.2,410.9,411.9
XS GIS Cut Line= 3
2136877.72033366644052.5394219972136910.73518539644807.996911464
 2137330.2180073645134.261328509
#Sta/Elev= 30
       0 1181.13    36.7 1159.74    88.7 1126.54   100.7 1117.32   108.7  1115.4
   164.8  1081.7   184.8 1071.41   208.8 1065.42   256.2 1045.71   272.9 1035.46
  309.491031.311     357  1028.7     385 1028.99  395.05 1031.31   433.1 1033.46
   486.3 1032.74   497.8 1034.25   553.2 1032.17   677.3 1031.95   745.4 1038.11
   864.4 1041.11  1072.2 1039.94  1116.4 1055.87  1137.2 1057.12  1175.1 1069.09
    1209 1082.57  1234.3 1089.89  1269.8 1108.58  1282.1 1110.89  1287.6 1113.77
#Mann= 6 ,-1,0
       0      .1       0  309.49    .045       0  395.05      .1       0
     600     .07       0  806.18      .1       0 1136.18     .06       0
Bank Sta=309.49,395.05
XS Rating Curve= 0 ,0
Exp/Cntr(USF)=0,0
Exp/Cntr=0.3,0.1
